--- EightenmC1.prj (project) ---

Proj Title=EightenmC1
Current Plan=p01
Default Exp/Contr=0,0
English Units
Geom File=g01
Flow File=f01
Plan File=p01
BEGIN DESCRIPTION:
AMEC Environment & Infrastructure, 2013
Projection: NAD 1983 State Plane West Virginia South FIPS 4702 (US Feet)
Vertical Datum: NAVD 1988
END DESCRIPTION:
DSS Export Rating Curves= 0
DSS Export Rating Curve Sorted= 0
DSS Export Volume Flow Curves= 0
DXF OffsetX= 0
DXF OffsetY= 0
DXF ScaleX= 0
DXF ScaleY= 0

--- EightenmC1.p01 (plan) ---

Plan Title=Floodplain
Program Version=4.00
Geom File=g01
Flow File=f01
K Sum by GR=0
Std Step Tol=0.01
Critical Tol=0.01
Num of Std Step Trials=20
Max Error Tol=0.3
Flow Tol Ratio=0.001
Split Flow NTrial=30
Split Flow Tol=0.02
Split Flow Ratio=0.02
Log Output Level=0
Friction Slope Method=1
Unsteady Friction Slope Method=2
Unsteady Bridges Friction Slope Method=1
Global Log Level=0
CheckData=False
Run HTab=0
Run UNet=0
Run PostProcess=0
UNET Theta=0
UNET Theta Warmup=0
UNET ZTol=0
UNET ZSATol=0
UNET MxIter=0
UNET MaxInSteps=0
UNET DtIC=0
UNET DtMin=0
UNET MaxCRTS=0
UNET WFStab=0
UNET SFStab=0
UNET WFX=0
UNET SFX=0
UNET DSS MLevel=0
UNET DZMax Abort=0
UNET Convert EG Bridges=0
UNET Use Existing IB Tables=0
UNET Froude Limit=0
UNET Froude Power=0
Write IC File=0
Echo Input=False
Echo Output=False
Write Detailed=0

--- EightenmC1.f01 (steady flow) ---

Flow Title=USGS Regress. Eqn. (2010) - Western-Plateaus
Program Version=4.10
Number of Profiles= 1
Profile Names=P100yr
River Rch & RM=EightenmC1,Main            ,106359.6
    1388
River Rch & RM=EightenmC1,Main            ,105305.6
    1588
River Rch & RM=EightenmC1,Main            ,103094.7
    1628
River Rch & RM=EightenmC1,Main            ,102076.1
    1788
River Rch & RM=EightenmC1,Main            ,101682.8
    1912
River Rch & RM=EightenmC1,Main            ,100412.1
    1946
River Rch & RM=EightenmC1,Main            ,98936.4
    1999
River Rch & RM=EightenmC1,Main            ,96375.6
    2258
River Rch & RM=EightenmC1,Main            ,94565.5
    2322
River Rch & RM=EightenmC1,Main            ,92899.9
    2339
River Rch & RM=EightenmC1,Main            ,91223.5
    2378
River Rch & RM=EightenmC1,Main            ,90424.8
    2428
River Rch & RM=EightenmC1,Main            ,88682.5
    2604
River Rch & RM=EightenmC1,Main            ,88103.3
    2612
River Rch & RM=EightenmC1,Main            ,86132.9
    2635
River Rch & RM=EightenmC1,Main            ,85533.4
    2639
River Rch & RM=EightenmC1,Main            ,84591.9
    2671
River Rch & RM=EightenmC1,Main            ,81631.3
    2861
River Rch & RM=EightenmC1,Main            ,81174.1
    3939
River Rch & RM=EightenmC1,Main            ,79297.6
    3978
River Rch & RM=EightenmC1,Main            ,77183.7
    3997
River Rch & RM=EightenmC1,Main            ,74206.4
    4047
River Rch & RM=EightenmC1,Main            ,69955
    4181
River Rch & RM=EightenmC1,Main            ,68814.9
    4188
River Rch & RM=EightenmC1,Main            ,67371.3
    4195
River Rch & RM=EightenmC1,Main            ,65982.3
    4234
River Rch & RM=EightenmC1,Main            ,63138.6
    4278
River Rch & RM=EightenmC1,Main            ,62132.5
    4285
River Rch & RM=EightenmC1,Main            ,60963.6
    6091
River Rch & RM=EightenmC1,Main            ,59035.5
    6289
River Rch & RM=EightenmC1,Main            ,56413.6
    6301
River Rch & RM=EightenmC1,Main            ,54544.9
    6314
River Rch & RM=EightenmC1,Main            ,51556.5
    6347
River Rch & RM=EightenmC1,Main            ,48799.5
    6403
River Rch & RM=EightenmC1,Main            ,46436.8
    6425
River Rch & RM=EightenmC1,Main            ,45472.2
    6727
River Rch & RM=EightenmC1,Main            ,44301.9
    6731
River Rch & RM=EightenmC1,Main            ,43092
    6743
River Rch & RM=EightenmC1,Main            ,41620
    7634
River Rch & RM=EightenmC1,Main            ,41143.9
    7636
River Rch & RM=EightenmC1,Main            ,40293.7
    7639
River Rch & RM=EightenmC1,Main            ,37988.7
    7646
River Rch & RM=EightenmC1,Main            ,35917.6
    7725
River Rch & RM=EightenmC1,Main            ,34410.6
    7777
River Rch & RM=EightenmC1,Main            ,31415.5
    7794
River Rch & RM=EightenmC1,Main            ,27137.4
    7872
River Rch & RM=EightenmC1,Main            ,24017.9
    7934
River Rch & RM=EightenmC1,Main            ,21565.8
    7962
River Rch & RM=EightenmC1,Main            ,21050.2
    8304
River Rch & RM=EightenmC1,Main            ,19753.6
    8309
River Rch & RM=EightenmC1,Main            ,18410.6
    8321
River Rch & RM=EightenmC1,Main            ,15454.3
    8435
River Rch & RM=EightenmC1,Main            ,13390.4
    8451
River Rch & RM=EightenmC1,Main            ,12291.9
    8457
River Rch & RM=EightenmC1,Main            ,10223.6
    8466
River Rch & RM=EightenmC1,Main            ,9629.6
    8927
River Rch & RM=EightenmC1,Main            ,7416
    8940
River Rch & RM=EightenmC1,Main            ,1983.3
    8997
River Rch & RM=EightenmC1,Main            ,420.8
    9262
River Rch & RM=EightenmC1,Main            ,0
    9265
Boundary for River Rch & Prof#=EightenmC1,Main            , 1
Up Type= 0
Dn Type= 1
Dn Known WS=579.88
DSS Import GetInterval= 0
DSS Import GetPeak= 0
DSS Import FillOption= 0

--- EightenmC1.g01 (geometry) ---

Geom Title=USGS 3m DEM
Program Version=4.10

River Reach=EightenmC1      ,Main
Reach XY= 30
     1758558.943        609032.9     1749190.709      602360.497
     1745924.867      602122.287     1745127.963      598806.726
     1742287.107      597847.015     1742069.008      596176.008
     1739879.338      596997.406     1739503.904      598763.899
     1738316.838      594119.801     1735287.324      593225.704
      1733142.36      594315.771     1733907.985      592987.646
     1731949.651      592599.625     1731694.443      591099.625
     1730319.443      593628.271     1729926.214      590966.813
     1726020.718       589331.61     1726413.891      591398.447
     1723682.988      591550.791     1724049.307      588312.944
     1721735.071      588800.791     1722931.252      587410.166
     1720125.696      586977.874     1718441.668       588408.43
     1716314.412      587275.531     1714186.373      590821.538
     1714919.012       593458.69     1712936.035      594324.038
     1712890.896      591002.857     1709238.506      591854.759

Type RM Length L Ch R = 1 ,106359.6,397.9,400.4,402.8
XS GIS Cut Line= 2
     1758510.391      608672.014     1758587.608      609395.908
#Sta/Elev= 30
       0   827.3      59  814.02   108.2  803.46     246  775.03   255.8  772.74
   265.6  769.29   275.5  764.11   324.6  733.66   334.5  727.89   344.3  723.52
   354.2  720.69   373.8  715.74   383.7     714   393.5  713.49     394  713.51
   403.4   713.8   442.7  716.21   511.6  719.89   541.1  721.72   560.8   723.2
   570.6  724.51   580.4   727.1   590.3  730.81   629.6  746.54   649.3  753.54
   659.1  756.44     669  758.39   678.8  759.04   688.6  758.77     728  757.02
#Mann= 3 , 0 , 0
       0      .1       0   354.2    .045       0     394     .08       0
Bank Sta=354.2,394
XS Rating Curve= 0 ,0
Exp/Cntr=0.3,0.1

Type RM Length L Ch R = 1 ,105959.2,223,232,241
XS GIS Cut Line= 2
     1758136.737       608729.46      1758174.13      609460.866
#Sta/Elev= 30
       0  817.09    58.6  801.12    78.1  796.19    97.6  792.47   205.1  774.18
   234.4  768.84   244.1  766.86   253.9  763.96   263.6  759.16   273.4  752.55
   302.7   729.9   312.5  723.39   322.2   719.3     332  717.24   354.3713.4371
   361.3  712.33   371.1   711.7   384.3712.1064   390.6  712.55   478.5  721.34
   488.2  722.67     498  724.36   507.8  726.52   517.5  729.79   527.3  734.49
   644.5  797.54   654.2  802.56     664     807   673.8  810.24   732.4  824.28
#Mann= 3 , 0 , 0
       0      .1       0   354.3    .045       0   384.3     .08       0
Bank Sta=354.3,384.3
XS Rating Curve= 0 ,0
Exp/Cntr=0.3,0.1

Type RM Length L Ch R = 1 ,105727.1,225.9,235.1,244.6
XS GIS Cut Line= 2
     1757962.793      608831.114     1757852.523      609583.622
#Sta/Elev= 30
       0  776.91    97.5     763   107.3   761.3     117  758.53   126.8  754.52
   175.5   732.3     195  723.63   214.5  715.39   224.3  712.07     234  710.72
   243.8  710.85   262.5712.5184   292.5  715.45     312  717.09   380.3  721.68
     390  722.23   409.5  722.82   419.3  723.51     429  725.06   448.5  728.99
   487.5  736.33   516.8  741.44   536.3  745.12   565.5  750.97   594.8  757.87
   614.3  762.02     624  763.77   692.3  770.75   731.3  774.05   760.5  777.14
#Mann= 3 , 0 , 0
       0      .1       0   224.3    .045       0   262.5     .08       0
Bank Sta=224.3,262.5
XS Rating Curve= 0 ,0
Exp/Cntr=0.3,0.1

Type RM Length L Ch R = 1 ,105492  ,164.8,186.4,207.2
XS GIS Cut Line= 2
     1757799.413      608767.142     1757536.602      609480.834
#Sta/Elev= 30
       0  768.39    48.8  759.62    87.8  751.25    97.5  748.68   107.3  744.18
   126.8  731.18   136.5  725.51   146.3  722.37     156  721.48   243.8  717.16
   253.5  716.17     273  711.88   282.8  710.46   292.5  710.35   313.6712.5441
   341.3  715.81   419.3  721.02     429  722.59   438.8  725.21     468  737.46
   487.5  746.92   516.8  762.86   575.3  796.98     585  802.11   594.8  806.44
   604.5  809.71   643.5  817.97   653.3   819.4   692.3  821.92   760.5  828.85
#Mann= 3 , 0 , 0
       0     .08       0   282.8    .045       0   313.6     .08       0
Bank Sta=282.8,313.6
XS Rating Curve= 0 ,0
Exp/Cntr=0.3,0.1

Type RM Length L Ch R = 1 ,105305.6,105.2,115.7,126.2
XS GIS Cut Line= 2
      1757746.87      608806.093     1757357.769      609178.522
#Sta/Elev= 30
       0  754.62    19.6  750.87    29.4  748.27    39.2  743.25      49  735.82
    58.8  727.89    68.6  721.55    78.3  718.92    97.9  718.16   195.9  716.22
   205.6  715.65     235  711.21   264.4  709.88     284  709.51   291.3  709.64
   303.6  710.64   313.4  712.51   323.2  715.15   342.8  720.27   352.6  723.09
   362.3  726.32   372.1  730.21   391.7  738.54   401.5  743.03   460.3  770.38
   489.6  784.52   499.4   788.9   509.2  792.74     519  796.01   538.6  801.92
#Mann= 3 , 0 , 0
       0     .08       0   291.3    .045       0   323.2     .08       0
Bank Sta=291.3,323.2
XS Rating Curve= 0 ,0
Exp/Cntr=0.3,0.1

Type RM Length L Ch R = 1 ,105189.9,179,188.5,198.5
XS GIS Cut Line= 2
     1757886.056      608678.952     1757169.925       609096.27
#Sta/Elev= 30
       0  792.42    29.2  788.67    68.3  778.86   224.3  749.81     234  746.25
   243.8  740.11   263.3  722.59     273  718.01   282.8  716.56   292.5  716.54
     351  718.44   380.3  717.88   399.8  716.02   438.8   708.8   448.6  708.62
   468.1  708.71   487.6  709.81   497.3  713.74   526.6  734.63   546.1     747
   565.6   756.9   585.1  765.02   614.3  775.13   633.8  780.69   653.3  785.26
   711.8  796.36   741.1  804.08   799.6  824.28   809.4  828.37   828.8  838.46
#Mann= 3 , 0 , 0
       0     .06       0   468.1    .045       0   497.3     .06       0
Bank Sta=468.1,497.3
XS Rating Curve= 0 ,0
Exp/Cntr=0.3,0.1

Type RM Length L Ch R = 1 ,105001.5,210.3,214.6,214
XS GIS Cut Line= 2
      1757689.19      608661.783     1757172.523      608822.379
#Sta/Elev= 30
       0  762.62    39.4  755.72    49.2   753.6      59  752.19    68.9  749.72
    78.7  741.01    88.5  727.54    98.4  717.96   108.2  714.94   147.6  713.66
   245.9  711.55   255.8  711.14   268.7  709.96   275.4  709.21   285.3   709.2
   295.1  712.02     305  717.69   314.8   724.1   324.6   729.7   334.5  734.83
   354.1  745.47     364  750.49   373.8  754.41   403.3  762.38   432.8  771.21
   452.5  776.73   462.4  779.75   511.5  796.83   521.4  800.45     541  808.12
#Mann= 3 , 0 , 0
       0     .06       0   268.7    .045       0   295.1     .06       0
Bank Sta=268.7,295.1
XS Rating Curve= 0 ,0
Exp/Cntr=0.3,0.1

Type RM Length L Ch R = 1 ,104786.9,433.7,413.2,394.5
XS GIS Cut Line= 2
     1757840.022      608480.554     1757082.368      608615.811
#Sta/Elev= 30
       0   796.4    68.2  779.24    97.4  775.03   107.2  773.11   233.8  741.75
   243.6  738.33   253.3  733.92   272.8   721.2   282.5  716.36   292.3  714.03
     302  713.25   331.2  713.21   350.7  712.14   366.6 709.178     380  706.83
   389.7   706.5   396.6706.8912   428.7  710.31   438.4  712.07   448.1  715.04
   457.9  719.66   487.1  738.87   496.8  744.46   506.6  748.16   535.8  751.66
     565     756   662.5  772.18   701.4  781.37   711.2  784.17   769.6  807.43
#Mann= 3 , 0 , 0
       0      .1       0   366.6    .045       0   396.6     .06       0
Bank Sta=366.6,396.6
XS Rating Curve= 0 ,0
Exp/Cntr=0.3,0.1

Type RM Length L Ch R = 1 ,104373.6,156.5,157.3,158
XS GIS Cut Line= 2
     1757611.256      607987.324     1757048.675      608451.578
#Sta/Elev= 30
       0  842.28    19.4  838.93    29.2  837.01    38.9  834.21    48.6  830.72
    58.4  826.86    97.2  810.68   136.2  794.98   155.6  786.87   243.1     749
   311.2  720.42   320.9  716.19   330.7  711.38   340.4  707.17   347.2705.6277
   350.1  704.97   359.8  705.03   377.2706.5844   525.2  720.34   544.6  721.84
   564.1   722.5   573.8  724.27   583.5  727.34   612.7  738.66   632.2  746.68
     671  764.02   680.8  767.44   690.5  769.93   700.2  772.11   729.4  778.26
#Mann= 3 , 0 , 0
       0      .1       0   347.2    .045       0   377.2     .06       0
Bank Sta=347.2,377.2
XS Rating Curve= 0 ,0
Exp/Cntr=0.3,0.1

Type RM Length L Ch R = 1 ,104216.4,129.1,129.1,129.1
XS GIS Cut Line= 2
     1757512.627      607872.856     1756943.594      608326.933
#Sta/Elev= 30
       0  836.81    39.4  821.03      59  812.97    78.7  805.15    88.5  801.39
   167.2  772.02   196.8  761.29   216.4  753.96   265.6  734.81   314.8  715.92
   334.5  707.55   344.3  704.79   348.2704.5615   354.2  704.21     364  705.08
   378.2706.8011   383.7  707.39   413.2  709.58   452.5  712.09   541.1  717.12
   590.3  719.54   600.1  721.28     610  724.61   619.8  729.09   639.5  738.78
     669  753.68   698.5  768.27   708.3  773.61   718.2  778.34     728  781.92
#Mann= 3 , 0 , 0
       0      .1       0   348.2    .045       0   378.2     .06       0
Bank Sta=348.2,378.2
XS Rating Curve= 0 ,0
Exp/Cntr=0.3,0.1

Type RM Length L Ch R = 1 ,104087.2,98.5,98.5,98.5
XS GIS Cut Line= 2
     1757418.856      607782.542     1756849.823      608236.619
#Sta/Elev= 30
       0  816.21     9.8  812.52   167.2  757.97   206.6  744.58   236.1  734.73
   275.5  721.87     305  713.34   324.6  705.48   328.5 704.826   334.5  703.82
   344.3  703.81   358.5705.1415   373.8  706.55   413.2  708.25   452.5  710.28
   511.6  712.69   541.1  714.32   560.8  715.95   580.4  717.98   600.1  720.11
     610  721.64   619.8  725.03   629.6   729.8     669  751.66   678.8  756.76
   688.6  760.89   698.5  764.08   708.3  767.01   718.2   769.6     728  771.67
#Mann= 3 , 0 , 0
       0      .1       0   328.5    .045       0   358.5     .06       0
Bank Sta=328.5,358.5
XS Rating Curve= 0 ,0
Exp/Cntr=0.3,0.1

Type RM Length L Ch R = 1 ,103988.8,155.1,155,155
XS GIS Cut Line= 2
     1757357.446      607705.585     1756788.413      608159.662
#Sta/Elev= 30
       0  807.96     118   768.3   157.4  755.22   186.9  745.64     246  727.11
   265.6  721.14     305  709.56   314.8  706.41   324.6  704.02   334.5  703.48
   344.3  705.51   354.2  707.84     364  709.08   373.8  709.34   403.4  709.31
   432.9  710.22   462.4   711.7   541.1   716.1   570.6  717.88   590.3  718.68
   600.1  718.58   619.8  719.23   639.5  719.24   649.3  719.45     669   721.5
   678.8  723.74   688.6   725.7   708.3  730.51   718.2  731.79     728  732.47
#Mann= 3 , 0 , 0
       0      .1       0   314.8    .045       0   354.2     .06       0
Bank Sta=314.8,354.2
XS Rating Curve= 0 ,0
Exp/Cntr=0.3,0.1

Type RM Length L Ch R = 1 ,103833.8,241.4,243.8,246.1
XS GIS Cut Line= 2
     1757270.624      607577.066     1756701.591      608031.143
#Sta/Elev= 30
       0  800.18    39.4  793.03      59  789.25    78.7   785.2    88.5  782.82
    98.4   779.8   108.2  776.13   157.4   756.6   177.1  749.06   186.9  745.49
   206.6  738.94   236.1  730.28   295.1  714.74   314.8  709.79   333.8704.6616
   344.3  702.95   354.2  702.72   363.8703.5527   403.4  708.52     423  710.07
   472.2  712.08   531.2  713.94   570.6   715.7   619.8  718.91   649.3  721.64
   659.1  723.11     669  725.81   688.6  732.02   718.2  739.94     728  742.95
#Mann= 3 , 0 , 0
       0      .1       0   333.8    .045       0   363.8     .06       0
Bank Sta=333.8,363.8
XS Rating Curve= 0 ,0
Exp/Cntr=0.3,0.1

Type RM Length L Ch R = 1 ,103590  ,499.5,495.3,467.4
XS GIS Cut Line= 2
     1757093.353      607430.509     1756500.927      607853.615
#Sta/Elev= 30
       0  767.27    39.4  761.98    78.7  756.13   108.2  750.99   127.9  746.97
   147.6     742   157.4  739.24   167.2  736.27   177.1  732.57   186.9  727.73
   206.6  717.46   216.4  713.27   226.3  710.56     246  706.83   255.8  704.68
   265.6  702.75   275.5  701.74   285.3  701.72   291.4  701.91   354.2   703.8
     423     705   462.4   706.2   491.9  706.72   501.7  707.22   531.2  711.53
   541.1  713.93   560.8  721.64     610  741.84   688.6  774.61     728  790.27
#Mann= 3 , 0 , 0
       0      .1       0   255.8    .045       0   291.4     .06       0
Bank Sta=255.8,291.4
XS Rating Curve= 0 ,0
Exp/Cntr=0.3,0.1

Type RM Length L Ch R = 1 ,103094.7,1018.5,1018.6,970.2
XS GIS Cut Line= 2
     1756961.925      606672.642     1756388.029       607690.52
#Sta/Elev= 30
       0  756.26    39.3  745.72    78.6  733.97    98.2  726.62   117.8  716.81
   127.6  713.13   137.5  711.67   206.2  711.83     275  709.61   343.7  708.95
   432.1  709.82   481.2  711.62   500.8  711.76   530.2  709.93   569.5  704.68
   589.2  700.67     599  699.79   628.4  699.58   687.4  699.49   765.9   700.2
   834.7  701.69   962.3  706.03     982   707.1   991.8  708.43  1001.6  711.48
  1011.4  716.01  1070.3  747.31    1090  756.31  1129.2  771.45  1168.5  784.03
#Mann= 3 , 0 , 0
       0      .1       0   569.5    .045       0   628.4     .08       0
Bank Sta=569.5,628.4
XS Rating Curve= 0 ,0
Exp/Cntr=0.3,0.1

Type RM Length L Ch R = 1 ,102076.1,354,393.3,413.1
XS GIS Cut Line= 2
     1756301.468      606699.232     1755879.644      607529.592
#Sta/Elev= 30
       0  751.18    19.6  745.95    29.4  743.92    39.2  742.63    78.4  739.02
   127.4  731.76   137.2   729.2   147.1   723.5   156.9  715.66   166.7  709.05
   176.5  706.01   313.7  699.75     402  697.22   421.6  696.21     451  696.45
     462695.8396   480.4  695.52     492696.1176   666.7  706.26   676.5  708.12
   686.3  710.77   725.5  722.84   754.9  732.66   813.7  753.27   823.5  755.94
   833.3  757.96   852.9     761   872.5  764.92   911.8  770.72   931.4  772.91
#Mann= 3 , 0 , 0
       0     .06       0     462    .045       0     492     .06       0
Bank Sta=462,492
XS Rating Curve= 0 ,0
Exp/Cntr=0.3,0.1

Type RM Length L Ch R = 1 ,101682.8,476.8,473.2,461.6
XS GIS Cut Line= 2
     1756203.015      606614.214     1755572.124      607053.846
#Sta/Elev= 30
       0  759.92    19.5  756.54    38.9  752.98    68.1   747.2    87.6  743.04
    97.3  740.14   107.1  735.51   116.8  729.41     146  709.17   155.7   703.9
   165.5  700.82   175.2  699.11   184.9  698.01   214.1  695.31   222.3694.8331
   233.6  694.49   252.3694.6862   311.5  695.81   360.2  697.19   389.4  698.15
     438  699.92   496.4   702.5   554.8  704.79   574.3  705.67   603.5  707.22
     623  708.45   710.6  714.74   749.5  716.95   759.2  717.74     769  719.39
#Mann= 3 , 0 , 0
       0      .1       0   222.3    .045       0   252.3     .08       0
Bank Sta=222.3,252.3
XS Rating Curve= 0 ,0
Exp/Cntr=0.3,0.1

Type RM Length L Ch R = 1 ,101209.6,398.6,391.4,389.5
XS GIS Cut Line= 2
      1755953.27      606222.547     1755448.236      606764.248
#Sta/Elev= 30
       0  786.61    29.2  778.42   116.9  754.34   126.7  751.55   136.4  747.95
   146.2  743.08   155.9  737.07   165.7  730.47   175.4  723.39   185.2  716.68
   194.9  710.84   204.6  706.41   214.4  703.72   253.4  697.34   272.9   693.8
   282.6  692.48   289.3692.1484   302.1  691.91   319.3692.0778   341.1  692.78
   370.3  694.22   399.5  695.05   516.5  699.46   545.7  700.78   584.7  703.04
   623.7  706.05   672.4  710.85   691.9  713.21   711.4  715.95   740.6  720.82
#Mann= 3 , 0 , 0
       0      .1       0   289.3    .045       0   319.3     .08       0
Bank Sta=289.3,319.3
XS Rating Curve= 0 ,0
Exp/Cntr=0.3,0.1

Type RM Length L Ch R = 1 ,100818.1,404.5,406,407
XS GIS Cut Line= 2
     1755667.774      605866.724     1755277.194      606483.192
#Sta/Elev= 30
       0  795.34    29.2  791.23    97.3   781.1     107  779.45   116.8  777.11
   126.5  774.45   155.7  765.85   165.4  762.86   175.2  759.44   204.3   748.6
     253  731.19   282.2  720.51   291.9  716.83   301.6  712.85   330.8  700.76
   340.6  696.51   350.3   693.2   351.1693.1027     360  692.02   369.8  691.94
   381.1692.2859   544.9  700.12   564.4  700.69   593.6  701.02     613  701.48
   671.4  703.86   681.1  704.36   690.9  705.07   700.6  706.01   729.8  709.53
#Mann= 3 , 0 , 0
       0      .1       0   351.1    .045       0   381.1     .08       0
Bank Sta=351.1,381.1
XS Rating Curve= 0 ,0
Exp/Cntr=0.3,0.1

Type RM Length L Ch R = 1 ,100412.1,394.7,396.5,397.2
XS GIS Cut Line= 2
     1755386.086      605596.444     1754980.072      606200.717
#Sta/Elev= 30
       0  763.89    19.7  763.82    29.5  763.31    98.4  758.82   127.9  756.54
   137.7  755.54   157.4  752.88   177.1  749.63   186.9  747.75   196.8   745.6
   206.6  742.92   226.3  736.84   236.1   733.4   265.6  722.31     305   707.8
   344.3  693.88     349692.8118   354.2  691.63     364  691.11   373.8  691.31
     379691.6672   442.7  696.26   531.2   702.1   590.3  706.57   639.5   711.4
   659.1  713.16   688.6  715.51   708.3  717.45   718.2  719.21     728  721.45
#Mann= 3 , 0 , 0
       0      .1       0     349    .045       0     379     .08       0
Bank Sta=349,379
XS Rating Curve= 0 ,0
Exp/Cntr=0.3,0.1

Type RM Length L Ch R = 1 ,100015.6,418.3,423.2,421
XS GIS Cut Line= 2
     1755175.118      605277.773      1754730.12      605900.825
#Sta/Elev= 30
       0  756.27    39.3   747.9    78.5  739.91   117.8  731.35   137.4   727.5
   157.1  723.96   176.7  721.02   186.5  719.86   235.6  714.92   255.2  712.44
   284.7  707.92   323.9  700.86   382.8  692.93   392.6  691.47   402.5  689.76
   407.3 689.187   412.3  688.59   422.1  688.25   437.3688.7855   452.3  689.52
   500.6  690.95   530.1  692.08   559.5  693.72   598.8   696.3   628.2  698.58
   696.9  704.62   736.2  707.81     746  708.81   755.8  710.56   765.6  713.54
#Mann= 3 , 0 , 0
       0     .06       0   407.3    .045       0   437.3     .08       0
Bank Sta=407.3,437.3
XS Rating Curve= 0 ,0
Exp/Cntr=0.3,0.1

Type RM Length L Ch R = 1 ,99592.4 ,232.6,220.6,208.4
XS GIS Cut Line= 2
     1754793.063      605187.435     1754348.066      605810.487
#Sta/Elev= 30
       0  763.53    68.7  747.56    98.2  740.33   147.2  727.78   176.7  720.95
   196.3  716.11   206.1  714.22     216  712.69   255.2  708.18   284.7  704.09
   314.1  698.84   343.6  692.97   363.2  688.55   366.8688.1276     373   687.4
   382.8   687.3   396.8688.0036   422.1  690.02   579.1  700.68     589  701.76
   608.6  705.31   618.4  706.93   628.2  708.05     638  709.94   647.9  713.18
   667.5  721.33   716.6  743.29   736.2  751.71     746  755.65   765.6  762.58
#Mann= 3 , 0 , 0
       0     .08       0   366.8    .045       0   396.8     .08       0
Bank Sta=366.8,396.8
XS Rating Curve= 0 ,0
Exp/Cntr=0.3,0.1

Type RM Length L Ch R = 1 ,99371.8 ,232.2,231.7,229.6
XS GIS Cut Line= 2
     1754490.615      605095.751     1754239.304      605801.542
#Sta/Elev= 30
       0  732.42     9.7  731.11    19.5  729.28    38.9  724.31    48.6  722.54
     107  717.07   116.8  715.65   126.5  713.17   155.7  703.06   165.4  700.65
   175.1  699.18   282.2  690.83   308.9687.9704   321.1  687.25   338.9 687.654
   496.2  695.46     506  696.16   515.7  697.75   525.4   700.2   544.9  705.78
   564.3  710.33   574.1  713.11   583.8  716.97   632.4  739.97   651.9  748.65
   661.6  752.67   681.1  760.05   700.6  766.89   729.7  776.34   749.2  782.13
#Mann= 3 , 0 , 0
       0     .06       0   308.9    .045       0   338.9     .08       0
Bank Sta=308.9,338.9
XS Rating Curve= 0 ,0
Exp/Cntr=0.3,0.1

Type RM Length L Ch R = 1 ,99140   ,191.9,203.6,215.8
XS GIS Cut Line= 2
     1754282.159      605026.564     1754056.042      605734.093
#Sta/Elev= 30
       0  711.47     9.8  712.03    19.6  712.16      88  711.05     127  710.89
   136.8  710.17   146.6  708.52   175.9  701.27   185.7  699.24   195.5  697.85
     215  696.68   244.3  695.55   293.2  694.39   332.3  693.09   371.4  690.79
   396.1688.1929   400.7   687.7   410.5  687.33   420.3  687.92   426.1688.8528
   459.4  694.77   469.1  697.85   488.7  707.03   498.4  710.99     518  715.92
   527.8  718.89   547.3   725.5   596.2  742.62   684.1  774.36   742.8   794.1
#Mann= 3 , 0 , 0
       0     .06       0   396.1    .045       0   426.1      .1       0
Bank Sta=396.1,426.1
XS Rating Curve= 0 ,0
Exp/Cntr=0.3,0.1

Type RM Length L Ch R = 1 ,98936.4 ,211.4,209,206.4
XS GIS Cut Line= 2
      1754175.39      605014.446      1753779.79      605638.725
#Sta/Elev= 30
       0  704.21    29.2  701.19    77.8  697.93    97.2  697.04   116.7  696.83
   145.9  697.09   184.8  696.62   204.2  695.97     282  692.22   330.6   690.5
   351.6688.0053   359.8  687.16   369.5  687.27   381.6688.8783   398.7  692.01
   408.4  694.37   418.2  697.95   437.6  706.88   447.3  710.57   457.1   712.9
   466.8  714.71   476.5  717.35     496  724.02   525.1  732.72   554.3   740.9
   593.2  751.24   622.4  758.29   680.7  770.45   709.9  776.14   739.1  781.34
#Mann= 3 , 0 , 0
       0     .06       0   351.6    .045       0   381.6      .1       0
Bank Sta=351.6,381.6
XS Rating Curve= 0 ,0
Exp/Cntr=0.3,0.1

Type RM Length L Ch R = 1 ,98727.4 ,351.1,334.7,315.3
XS GIS Cut Line= 2
     1753990.708       604912.52     1753610.213      605546.118
#Sta/Elev= 30
       0  706.43     9.7  705.26    19.4  704.49    48.6   703.1   126.4  695.88
   194.5  690.88   213.9  689.82   243.1  688.66   327.6686.3326   340.4  686.26
   350.1  686.54   357.6687.1895   379.3  689.35   457.1  695.78   466.8  696.84
   476.5  698.57   486.2   701.4   505.7  709.68   525.1  714.08   534.8  716.96
   544.6  720.88     564  729.11   573.8  732.29   583.5  734.68   593.2  736.15
   602.9   737.2   612.6  737.56   641.8  737.98   709.9  739.67   739.1  739.91
#Mann= 3 , 0 , 0
       0     .08       0   327.6    .045       0   357.6     .08       0
Bank Sta=327.6,357.6
XS Rating Curve= 0 ,0
Exp/Cntr=0.3,0.1

Type RM Length L Ch R = 1 ,98392.7 ,388.1,390.5,393.5
XS GIS Cut Line= 4
      1753750.31      604600.388      1753650.48      605066.171
     1753662.294      605166.454     1753516.382      605562.397
#Sta/Elev= 30
       0  743.14    19.4  742.98    48.6  744.63    87.5  744.79   116.7  742.87
   136.1  740.01   155.6     735     175  728.54     243  702.84   262.5  695.92
   272.2  693.32   291.6  688.94   301.4  686.99   308.3686.2786   320.8   685.8
   338.3 686.442   476.4  692.15     559  692.42   675.5  694.23   704.9  695.16
   724.5  696.16     754  698.29   783.4  702.36   793.2  702.61   842.3  701.78
   891.4  702.13   930.6     703   950.2  703.93   989.5  709.46   999.3  709.99
#Mann= 3 , 0 , 0
       0      .1       0   308.3    .045       0   338.3     .08       0
Bank Sta=308.3,338.3
XS Rating Curve= 0 ,0
Exp/Cntr=0.3,0.1

Type RM Length L Ch R = 1 ,98002.3 ,369.8,414.5,454.1
XS GIS Cut Line= 2
     1753352.584      604710.389     1753215.234      605431.021
#Sta/Elev= 30
       0  725.73    29.3  726.09    68.5  727.03      88  726.89    97.8  726.32
   127.2  722.99   136.9  719.89   146.7  711.45   156.5   701.2   166.3  694.68
   176.1  691.79   205.4  686.09   210.9685.3099   215.2   684.7     225  684.24
   240.9684.5424   332.6  686.35   352.1  687.15   371.7  688.31     401  690.38
   498.8  698.81   586.9   705.4   596.7  706.47   606.4  708.75   616.2  712.33
   655.4  728.88   674.9   736.4   704.3   746.6     714  749.79   733.6  755.79
#Mann= 3 , 0 , 0
       0      .1       0   210.9    .045       0   240.9     .06       0
Bank Sta=210.9,240.9
XS Rating Curve= 0 ,0
Exp/Cntr=0.3,0.1

Type RM Length L Ch R = 1 ,97587.8 ,346.1,335.1,323.9
XS GIS Cut Line= 2
     1753339.487      604669.405     1752671.059      605005.784
#Sta/Elev= 30
       0   723.1    48.6  721.09   116.6   719.1     136  718.12   145.8  715.76
   155.5  709.78   165.2  702.14   174.9  696.18   184.6  693.16   194.4  691.98
   213.8  690.81   427.1682.8875   437.3  682.62     447   682.7   457.1683.6222
   485.9  689.81   495.6  694.31   505.3  701.08   524.8  716.13   544.2  730.61
   553.9  736.96   563.6  740.77   573.4   742.3   583.1  743.08   612.2  745.05
   651.1  747.05   699.7  751.16   728.9   753.9   738.6  754.48   748.3  754.27
#Mann= 3 , 0 , 0
       0     .06       0   427.1    .045       0   457.1      .1       0
Bank Sta=427.1,457.1
XS Rating Curve= 0 ,0
Exp/Cntr=0.3,0.1

Type RM Length L Ch R = 1 ,97252.7 ,512.1,517.1,517.7
XS GIS Cut Line= 3
     1753085.749      604337.528     1752596.258      604734.092
     1752445.626      605166.502
#Sta/Elev= 30
       0  693.83    38.8  692.64    87.2   690.4   145.4  690.94   184.2  690.27
   300.4  685.42   353.7682.2626   368.3  681.82   383.7682.6689   426.4  687.72
     504  693.42   513.7  695.27   523.4  697.94   552.4  708.39   562.1  710.31
   581.5  712.47   610.6  716.52   620.3  717.16     630  716.87   639.7  718.84
   649.5  719.96   688.4  720.75   746.9  719.72   795.6  716.68     854  714.53
   961.2  716.02   990.4  717.22  1009.9  718.71  1048.9  723.95  1087.9  730.88
#Mann= 3 , 0 , 0
       0     .06       0   353.7    .045       0   383.7      .1       0
Bank Sta=353.7,383.7
XS Rating Curve= 0 ,0
Exp/Cntr=0.3,0.1

Type RM Length L Ch R = 1 ,96735.6 ,373.8,360,346.2
XS GIS Cut Line= 2
     1752843.188      603948.401     1751914.254      604687.142
#Sta/Elev= 30
       0  731.11    98.1  723.63   166.8  720.07   186.4  719.79   225.6   720.8
   284.5  720.67   313.9  719.53   333.5  717.79   353.1  712.88   362.9  709.13
     412  684.64   421.8  682.17   428.8  681.47   431.6  681.19   458.8681.6704
   578.7  685.74   637.6  688.37   647.4  689.71   676.8   696.4   686.6  697.94
   696.4  700.46   745.5  721.45   774.9   732.7   931.8  789.87   980.9  806.32
  1029.9   820.7  1098.6   838.4  1118.2  842.74  1167.2  851.36  1186.9  856.46
#Mann= 3 , 0 , 0
       0      .1       0   428.8    .045       0   458.8      .1       0
Bank Sta=428.8,458.8
XS Rating Curve= 0 ,0
Exp/Cntr=0.3,0.1

Type RM Length L Ch R = 1 ,96375.6 ,360.4,330.3,298.5
XS GIS Cut Line= 2
     1752443.431      603733.932     1751993.044      604306.596
#Sta/Elev= 30
       0  751.37   116.6  739.55   126.3  738.34     136  736.24   155.4  728.28
   223.4  696.67   233.1  692.68   242.8  689.73   252.6  688.39   262.3  687.85
   388.6   683.7   436.2 681.452   446.8  680.97   456.6  681.44   466.2683.4986
   485.7  691.06   495.4  694.08   505.1  695.54     544  695.49   563.4  697.32
   573.1  699.75   592.6  707.91     612  718.98   631.4  734.36   660.6     756
   670.3  761.01   689.7  770.08   699.4  772.46   709.1  773.74   728.6   777.9
#Mann= 3 , 0 , 0
       0     .06       0   436.2    .045       0   466.2      .1       0
Bank Sta=436.2,466.2
XS Rating Curve= 0 ,0
Exp/Cntr=0.3,0.1

Type RM Length L Ch R = 1 ,96045.3 ,522.8,523.5,522.3
XS GIS Cut Line= 2
     1751857.235      603536.411     1751871.231      604281.468
#Sta/Elev= 30
       0   749.6    19.6  741.36    68.6  720.14    88.2  711.81      98  707.84
   127.5  696.38   147.1  687.61   156.9  685.25   186.3  684.33   225.5  682.87
   274.5  681.84   333.4  681.08   412.5680.6714   431.4   680.5   441.2  681.34
   442.5681.7167     451  684.18   460.8  688.17   470.6  691.77   480.4  694.85
   490.3  697.48   500.1   699.8   509.9  702.47   568.7   720.8   598.1  730.42
   617.7  737.18   637.3  744.15   666.8  754.86   725.6  776.55   745.2  783.51
#Mann= 3 , 0 , 0
       0     .06       0   412.5    .045       0   442.5      .1       0
Bank Sta=412.5,442.5
XS Rating Curve= 0 ,0
Exp/Cntr=0.3,0.1

Type RM Length L Ch R = 1 ,95521.8 ,457.9,470.5,456.1
XS GIS Cut Line= 2
     1751414.335      603504.666     1751440.771      604272.601
#Sta/Elev= 30
       0  782.79    19.4  778.35    48.6  771.98    68.1   768.1    97.3  762.66
     107  759.93   116.7  756.29   155.6  739.86   194.5  723.73   262.6  695.88
   282.1   688.1   291.8   684.6   301.5  681.88   311.2  679.91     322678.4561
   330.7   677.9   340.4  677.86     352678.2095   389.1  680.92     428   684.1
   515.5     692   525.2  693.17     535  695.12   544.7  697.99   573.9     708
     603  718.72   622.5  726.34   680.8  749.66     710  761.01   768.4  783.21
#Mann= 3 , 0 , 0
       0      .1       0     322    .045       0     352      .1       0
Bank Sta=322,352
XS Rating Curve= 0 ,0
Exp/Cntr=0.3,0.1

Type RM Length L Ch R = 1 ,95051.3 ,465.6,485.7,494.4
XS GIS Cut Line= 2
      1751029.07      603596.106     1751097.284      604352.645
#Sta/Elev= 30
       0  741.86      39   732.2    77.9  721.85   116.9  711.06   146.1   702.8
   175.3  694.41   204.5  685.78   214.2  683.63     224  682.49   233.7   681.9
   262.9  680.43   301.9  678.96   350.6  677.82   429.7676.7051   438.2   676.6
     448  676.82   457.7   678.2   459.7678.8598   467.4   681.4   486.9  690.17
   535.6  711.09   564.8  723.36   613.5  743.58     633  751.58   642.8   755.3
   652.5  758.21   662.2  759.77     672  760.21   720.6  760.77   759.6  761.53
#Mann= 3 , 0 , 0
       0      .1       0   429.7    .045       0   459.7      .1       0
Bank Sta=429.7,459.7
XS Rating Curve= 0 ,0
Exp/Cntr=0.3,0.1

Type RM Length L Ch R = 1 ,94565.5 ,562.4,589.4,615.3
XS GIS Cut Line= 2
     1750710.855       603586.46      1750596.82       604379.49
#Sta/Elev= 30
       0  753.74    19.5   748.5    29.3  745.46    48.8  738.53    78.2  726.38
   117.2  708.87   136.8  700.46   166.1  689.01   175.9  685.97   185.6  684.26
     254  679.47     342  676.47   419.7674.6262   429.9  674.53   439.7  674.62
   449.7675.3599   459.2  676.94   478.8  681.04   527.6  690.12   537.4  692.33
   547.2  695.35   586.2  711.21     596  714.96   615.6  721.62   644.9  730.91
   683.9  744.34   713.2  754.03   732.8  761.12   762.1  772.46   801.2  786.08
#Mann= 3 , 0 , 0
       0      .1       0   419.7    .045       0   449.7      .1       0
Bank Sta=419.7,449.7
XS Rating Curve= 0 ,0
Exp/Cntr=0.3,0.1

Type RM Length L Ch R = 1 ,93976.2 ,343.9,352,358.9
XS GIS Cut Line= 2
     1750555.936      603447.639     1750030.799      603965.191
#Sta/Elev= 30
       0  766.02    19.7  759.69    49.2  751.95   147.5  720.83   167.1  713.98
   206.4  699.26   226.1  692.42   245.8  686.25   265.4  680.68   275.3  678.34
   285.1  676.66   294.9  675.75   365.9673.9433   373.6  673.78   383.4  673.78
   395.9674.3546   452.2  680.58   491.5  685.52   501.4  688.87   511.2  693.27
   530.9  702.68   589.8  731.65   619.3  745.54     639  754.05   648.8   757.4
   658.7  759.57   668.5  759.97   688.2  758.67   717.6  755.95   737.3   754.9
#Mann= 3 , 0 , 0
       0      .1       0   365.9    .045       0   395.9      .1       0
Bank Sta=365.9,395.9
XS Rating Curve= 0 ,0
Exp/Cntr=0.3,0.1

Type RM Length L Ch R = 1 ,93624.2 ,399.2,366.8,335
XS GIS Cut Line= 2
     1750417.904      603175.184     1749839.399      603631.791
#Sta/Elev= 30
       0  778.73    29.5  770.61    49.1  767.61    68.8   766.2   117.9  764.23
   147.4  762.34     167  760.26   176.9  758.59   186.7  756.16   196.5  752.32
   206.4  747.67   294.8  703.19   334.1  684.65   343.9  679.55   353.8  675.66
   357.8674.9539   363.6  673.93   373.4  673.75   387.8674.2079   481.5  677.24
   491.3  678.84   501.2  682.37   530.6   696.8   540.5   699.7   550.3  701.25
   579.8  703.38   619.1  707.79   687.9  716.74   697.7  718.66     737  728.16
#Mann= 3 , 0 , 0
       0      .1       0   357.8    .045       0   387.8     .08       0
Bank Sta=357.8,387.8
XS Rating Curve= 0 ,0
Exp/Cntr=0.3,0.1

Type RM Length L Ch R = 1 ,93257.3 ,335,357.5,375.5
XS GIS Cut Line= 2
     1749908.068      602859.285     1749763.216      603631.033
#Sta/Elev= 30
       0  764.26    39.3  759.35    58.9   757.6    78.5  756.32     108  752.66
   137.4  747.82   196.3  736.47   235.6     730   245.4  726.98   255.2  722.57
   274.8  712.03   304.3  695.49   314.1  689.76   333.7   677.4   341.7674.5673
   343.5  673.93   353.4  673.18   371.7673.9736   471.1  677.98   510.4  680.32
     530  682.18   579.1  689.95   598.7  693.52   608.6  695.68   647.8   706.2
   657.6  707.92   667.4  709.04   677.3  710.85   726.3  725.72   785.2  743.09
#Mann= 3 , 0 , 0
       0      .1       0   341.7    .045       0   371.7     .06       0
Bank Sta=341.7,371.7
XS Rating Curve= 0 ,0
Exp/Cntr=0.3,0.1

Type RM Length L Ch R = 1 ,92899.9 ,237.7,282.6,326
XS GIS Cut Line= 2
     1749675.936      603073.388     1749408.106      603464.947
#Sta/Elev= 30
       0  702.78    19.4  699.24    38.7   696.1    48.4  694.73    67.8  692.44
   164.6  682.89   193.6  680.87     213  680.08   222.7  679.48   232.4  678.31
   251.7  675.31   273.8672.4255   280.8  671.61   290.4  671.16   300.1  672.13
   303.8673.7244   309.8  676.31   319.5  683.45   348.5   707.6   358.2  714.31
   367.9  718.71   377.6  723.57   387.3  731.91   396.9  741.98   406.6  749.49
   416.3  753.72     426  756.07     455  761.14   464.7  763.68   474.4  767.06
#Mann= 3 , 0 , 0
       0      .1       0   273.8    .045       0   303.8      .1       0
Bank Sta=273.8,303.8
XS Rating Curve= 0 ,0
Exp/Cntr=0.3,0.1

Type RM Length L Ch R = 1 ,92617.3 ,299.5,280.7,261.9
XS GIS Cut Line= 2
     1749685.912       603051.58     1749305.276      603047.106
#Sta/Elev= 30
       0  706.87     9.8  705.09    19.5  703.14    29.3  700.94    58.6  693.61
    68.3   691.4    87.8  687.33   136.6  677.87   146.4  676.05   165.9   672.7
   170.9672.0724   175.7  671.47   185.4  671.11   195.2  672.02   200.9673.4043
     205   674.4   214.7  677.39   224.5  680.15   234.2  682.61     244  684.86
   263.5  688.95   273.3  690.79   292.8  694.23   302.6  695.86   312.3  697.43
   322.1  698.84   331.9  699.83   351.4  700.73   361.1  701.33   380.7  702.84
#Mann= 3 , 0 , 0
       0      .1       0   170.9    .045       0   200.9     .08       0
Bank Sta=170.9,200.9
XS Rating Curve= 0 ,0
Exp/Cntr=0.3,0.1

Type RM Length L Ch R = 1 ,92336.6 ,277.8,270.9,262.9
XS GIS Cut Line= 2
     1749850.594      602611.693     1749119.085      602917.569
#Sta/Elev= 30
       0  788.32    19.6  782.57    78.3  768.33    88.1  766.37    97.9  764.77
   166.4   754.9   176.2   753.3   195.8  748.98   205.6  746.24   254.5   729.6
   264.3  726.69   274.1     724   332.8  709.29   352.4  704.05   362.2  701.16
     372  697.87   381.8  694.31   401.3  686.85   411.1  682.59   420.9  677.46
   430.7  673.02   433.6672.3956   440.5  670.91   450.3  670.73   463.6671.5136
   499.2  673.77   626.5   680.6   743.9  685.66   773.3  686.41   792.9  687.42
#Mann= 3 , 0 , 0
       0      .1       0   433.6    .045       0   463.6     .06       0
Bank Sta=433.6,463.6
XS Rating Curve= 0 ,0
Exp/Cntr=0.3,0.1

Type RM Length L Ch R = 1 ,92065.7 ,523.4,454.9,381.9
XS GIS Cut Line= 3
     1749628.032      602352.956     1749194.054      602625.684
     1749058.745      602996.179
#Sta/Elev= 30
       0  776.73    19.3  773.85      58  767.19    77.4  764.58   106.4  762.34
   164.4  759.99   174.1  759.31   183.8  757.62   193.4  754.22   203.1  749.29
   212.8  743.61   232.1  731.27   280.5  697.53   290.1  691.44   319.1  674.27
   328.8  670.98   338.5  670.46   366.6  672.85   396.5  674.41   464.2  676.71
   560.7  678.85   637.6  679.52   676.1  680.24   753.1  682.85   781.9  684.24
   801.2  685.61     830  688.67   849.3  691.17   878.1   695.9     907  701.82
#Mann= 3 , 0 , 0
       0      .1       0   319.1    .045       0   366.6     .06       0
Bank Sta=319.1,366.6
XS Rating Curve= 0 ,0
Exp/Cntr=0.3,0.1

Type RM Length L Ch R = 1 ,91610.8 ,364.9,387.3,410
XS GIS Cut Line= 3
     1748821.856      602132.927     1749146.005      602659.033
     1749013.589      603037.855
#Sta/Elev= 30
       0  798.05    39.2  792.74    78.5  785.97   137.3  773.68   147.1  771.28
   156.9  768.32   166.8  764.39   176.6  759.29   186.4  753.53   225.6  728.23
   264.8  702.27   274.6  696.32   294.3  685.84   313.9  674.53   323.7  671.07
   333.5  669.87   369.7  670.29     412  670.97   470.8  672.47   529.7  674.51
     618   678.2   784.3  681.76   833.3  683.56   862.6  686.93     892  688.67
   921.4  691.42   960.5   697.1   999.7  704.58  1009.5  705.76  1019.2  706.38
#Mann= 3 , 0 , 0
       0      .1       0   323.7    .045       0   369.7     .06       0
Bank Sta=323.7,369.7
XS Rating Curve= 0 ,0
Exp/Cntr=0.3,0.1

Type RM Length L Ch R = 1 ,91223.5 ,401.6,446.1,490.5
XS GIS Cut Line= 2
     1748730.531      602157.573     1748784.926      603048.537
#Sta/Elev= 30
       0  771.51    19.6  765.94    39.2  760.09    88.3  744.54   137.3  729.95
   245.2  699.11   304.1  681.92   313.9  679.88   323.7  678.64   333.5  677.76
   392.4  673.34     412  672.06   431.6  671.05   470.8  669.44   549.3  666.78
   568.9  666.27   578.7  666.38   590.4  667.37   608.2  669.73     618  670.66
     667  674.05   735.7  679.53   765.1  681.59   774.9  683.06   784.7  685.49
   794.5  688.25   804.3  690.57   814.2  692.28   863.2  698.74   892.6  701.77
#Mann= 3 , 0 , 0
       0     .06       0   549.3    .045       0   590.4     .06       0
Bank Sta=549.3,590.4
XS Rating Curve= 0 ,0
Exp/Cntr=0.3,0.1

Type RM Length L Ch R = 1 ,90777.4 ,361.9,352.6,342.4
XS GIS Cut Line= 2
     1748710.587      602327.206     1748008.664      602853.474
#Sta/Elev= 30
       0     718    29.2  711.03    58.5  705.05   107.2  694.57   126.7     690
     156  682.56   165.7   680.4   175.5  678.93   331.4  670.02   370.4  668.16
   411.7  666.61   448.4  665.58   458.2  665.92   467.9  668.07   471.7  670.93
   477.6  675.37   487.4  685.17   497.1  692.48   506.9  696.39   516.6  699.64
   536.1  708.32   545.9   711.1   555.6  712.41   604.4  716.06   643.4  719.52
   711.6   726.3   750.6  729.61   828.6  737.61   848.1  739.18   877.3  740.92
#Mann= 3 , 0 , 0
       0     .06       0   411.7    .045       0   471.7      .1       0
Bank Sta=411.7,471.7
XS Rating Curve= 0 ,0
Exp/Cntr=0.3,0.1

Type RM Length L Ch R = 1 ,90424.8 ,372.2,255.8,234.4
XS GIS Cut Line= 2
     1748543.068      601982.528     1748030.991      602555.755
#Sta/Elev= 30
       0  768.17    29.2  756.06    87.6  730.19   116.8  717.96   136.2  710.47
   155.7  703.58   184.9  694.56     214  687.14   233.5  683.19   243.2  681.73
   262.7  679.36   291.9  677.77   301.6  676.79     360  668.39   369.7  666.78
   379.5  665.82   389.2  665.55   408.6  666.21   525.4  671.45   535.1  671.94
   544.9  673.04   554.6  675.92     574  685.18   583.8   688.8   603.2   693.1
   622.7  699.59   632.4  701.99   642.2  703.23   700.5  708.02   768.6  711.64
#Mann= 3 , 0 , 0
       0     .06       0     360    .045       0   408.6     .06       0
Bank Sta=360,408.6
XS Rating Curve= 0 ,0
Exp/Cntr=0.3,0.1

Type RM Length L Ch R = 1 ,90169.1 ,157.2,229.3,202.6
XS GIS Cut Line= 4
     1748027.473      601568.999     1748102.901      602133.775
     1747998.029      602415.402     1747913.816      602641.552
#Sta/Elev= 30
       0  780.38    39.3  774.84    58.9  771.48    88.4  765.13   108.1  759.63
   157.2   742.4   206.3  726.66   324.2  679.37     334  675.57   343.8   672.7
   353.7  671.66   373.3   671.4   442.1  667.23   530.5   665.8   550.1  665.36
   569.8  665.65   590.5  666.74   744.3  670.97     754  672.41   763.7  675.22
   783.1  682.34   792.8   684.5   812.1  687.62   850.9  697.01   899.3  703.61
   928.2  706.74   986.1  710.52  1034.4  712.88    1073   713.7  1111.6  713.48
#Mann= 3 , 0 , 0
       0      .1       0   530.5    .045       0   590.5     .06       0
Bank Sta=530.5,590.5
XS Rating Curve= 0 ,0
Exp/Cntr=0.3,0.1

Type RM Length L Ch R = 1 ,89939.8 ,137.9,159.5,183.7
XS GIS Cut Line= 4
     1747929.884      601582.033     1748002.059      602122.449
     1747905.764      602381.045      1747821.55      602607.195
#Sta/Elev= 30
       0  767.01    38.9  763.86    87.6  756.94   126.6  749.12   165.5  738.89
     185  731.75   204.5  723.72   214.2   719.4   243.4  704.48   253.1  700.71
   272.6  695.02   282.3  690.99   321.3  671.94   332.2   667.7   340.8  665.86
   360.2  665.16   392.2  665.28   583.3  667.24   659.4   668.8   687.9  670.21
   716.5  673.86     745  679.85   773.6   684.9   811.6  694.64   869.4  701.96
     908  708.04     937  709.68   985.3  709.92  1014.2   709.6  1062.5  707.56
#Mann= 3 , 0 , 0
       0      .1       0   332.2    .045       0   392.2     .06       0
Bank Sta=332.2,392.2
XS Rating Curve= 0 ,0
Exp/Cntr=0.3,0.1

Type RM Length L Ch R = 1 ,89780.3 ,293.7,293.8,294
XS GIS Cut Line= 3
     1747899.098      601574.239     1747742.545      602285.228
     1747698.191      602486.663
#Sta/Elev= 30
       0   763.5     9.8  763.24    19.7  762.57    39.4  760.25      59  757.34
    78.7  753.59    98.4  748.93   118.1  743.65   147.6  735.36   186.9  723.87
   206.6  719.22   216.4  716.64   226.3  712.15   236.1  706.55   275.5  683.33
   286.2     676   295.1  669.74     305  665.75   314.8  665.01   346.2  665.67
   452.6  666.54   541.1  667.65   659.2  669.79   698.5  669.64   737.8  671.77
   757.5  672.26     787  672.52   836.1   674.1   914.6   674.2   934.3  673.83
#Mann= 3 , 0 , 0
       0      .1       0   286.2    .045       0   346.2     .06       0
Bank Sta=286.2,346.2
XS Rating Curve= 0 ,0
Exp/Cntr=0.3,0.1

Type RM Length L Ch R = 1 ,89486.5 ,364.9,362.6,357.3
XS GIS Cut Line= 3
     1747620.375      601482.173     1747463.822      602193.163
     1747419.468      602394.597
#Sta/Elev= 30
       0  775.33     9.8  773.37    39.4  768.11      59  765.23    68.9  763.56
    78.7  761.32   118.1  750.68   147.6  742.28   167.2  736.23   186.9  729.33
   216.4  718.42   226.3  714.39   265.6  696.79   285.3  688.29   333.8   668.6
   344.3  664.79   354.2  662.86     364  662.42   393.8  662.65   472.2  664.46
   550.9  665.94     610   668.1   688.7  670.32   777.1  673.44   816.4  674.62
   826.2  675.46   836.1  676.86   845.9  678.82   865.5  683.68   934.3  702.18
#Mann= 3 , 0 , 0
       0      .1       0   333.8    .045       0   393.8     .06       0
Bank Sta=333.8,393.8
XS Rating Curve= 0 ,0
Exp/Cntr=0.3,0.1

Type RM Length L Ch R = 1 ,89123.9 ,452.9,441.4,429.3
XS GIS Cut Line= 3
     1747228.499      601491.847     1747125.932      602213.833
     1747122.398      602238.709
#Sta/Elev= 30
       0  728.26    29.2  721.78    87.5  708.69   116.7   702.3   136.1  697.97
   204.2  683.36   272.2  668.98   289.4  664.91   291.7  664.36   301.4  662.87
   311.1  662.44   320.9  662.41   340.3  662.58   349.4  662.78   379.2   663.5
   388.9  663.92   408.4  664.95   447.3  666.68   476.4   668.2   505.6  669.96
     525  671.25   554.2  673.33   602.8  677.04   670.9  682.51   700.1  684.76
   719.5   686.4   729.2  687.01   737.6  687.84     746  689.42   754.4   691.8
#Mann= 3 , 0 , 0
       0      .1       0   289.4    .045       0   349.4     .06       0
Bank Sta=289.4,349.4
XS Rating Curve= 0 ,0
Exp/Cntr=0.3,0.1

Type RM Length L Ch R = 1 ,88682.5 ,601.5,579.2,555.4
XS GIS Cut Line= 3
     1746765.652      601210.154     1746858.011      601964.978
     1746894.152      602260.356
#Sta/Elev= 30
       0  761.61      39  754.68    58.5  750.58   126.7   734.8     195  718.14
   204.7   715.4   214.5  712.14   243.7  700.64   263.2  693.49   282.7  687.55
   331.5  674.72     352   668.3   360.7  665.19   370.5  662.96   380.2   662.4
     412   662.4   448.5  662.48   526.5  663.57   643.5  664.76   731.2  666.18
   808.4  667.84   923.6  669.65   933.2  670.18     962  673.18   990.8  675.46
  1000.4  676.52    1010  678.66  1019.6  681.66  1038.8  688.31    1058  695.34
#Mann= 3 , 0 , 0
       0      .1       0     352    .045       0     412     .06       0
Bank Sta=352,412
XS Rating Curve= 0 ,0
Exp/Cntr=0.3,0.1

Type RM Length L Ch R = 1 ,88103.3 ,331,409.4,456.7
XS GIS Cut Line= 2
     1746207.075      601604.393     1746633.724      602251.256
#Sta/Elev= 30
       0  737.29    68.7  723.53    88.3  718.87    98.1  716.08   127.5  706.78
   147.1  699.88   196.2   679.8   215.8  672.43   236.9  665.01   245.2  662.28
     255  660.06   264.8  659.32   274.6  659.54   296.9  661.89   304.1  662.19
   333.5  661.56   362.9  661.52     461  663.38   490.4  664.19   519.9  664.48
   559.1   666.9   627.8     670   637.6  671.36   647.4  673.67   657.2  674.76
   676.8  673.45   686.6  673.33     716  674.47   735.7  676.49   774.9  677.46
#Mann= 3 , 0 , 0
       0      .1       0   236.9    .045       0   296.9     .06       0
Bank Sta=236.9,296.9
XS Rating Curve= 0 ,0
Exp/Cntr=0.3,0.1

Type RM Length L Ch R = 1 ,87693.9 ,597.9,578.5,585
XS GIS Cut Line= 2
     1746212.135      601472.064     1746048.257      602480.375
#Sta/Elev= 30
       0  787.45     9.8   784.1    29.5  776.29    88.4   751.8   137.5  733.81
   235.7   700.2   304.5  675.46   314.3  672.87   324.1     671   343.8  665.17
   353.6  663.48   363.4  662.95   481.3  660.48   540.2  660.18     609   661.2
   628.6  660.85   654.8  659.77   687.6  658.44   697.4  658.71   707.2  659.46
   714.8  660.62   726.9  663.27   766.2  673.71   795.6  682.96   815.3  690.04
   864.4   710.5   913.5  733.01   952.8  750.13   982.2  761.62  1021.5  775.59
#Mann= 3 , 0 , 0
       0     .06       0   654.8    .045       0   714.8      .1       0
Bank Sta=654.8,714.8
XS Rating Curve= 0 ,0
Exp/Cntr=0.3,0.1
