HEC-RAS study EightenmC1.prj: EightenmC1

--- EightenmC1.g01 (geometry) --- (continued)

Type RM Length L Ch R = 1 ,87115.5 ,394.4,396.1,361.2
XS GIS Cut Line= 2
     1746067.619      601428.738     1745512.726      602069.004
#Sta/Elev= 30
       0  775.23    29.2  763.89    58.4  752.82     185  707.01   243.5  685.99
   253.2  682.15   262.9   678.1   272.7  673.85   282.4   669.2   292.2  665.26
   301.9  663.23   311.6  662.69   463.4  658.02   486.9  657.47   496.7  657.61
   506.4  657.93   516.2  658.58   523.4  659.25   535.6   660.7   574.6  666.55
   613.5  671.48   623.3  672.99     633  674.88   642.8  677.36   652.5  680.86
     672  689.57   681.7  693.58   691.4  697.11   788.8  730.94   847.3  752.04
#Mann= 3 , 0 , 0
       0     .06       0   463.4    .045       0   523.4      .1       0
Bank Sta=463.4,523.4
XS Rating Curve= 0 ,0
Exp/Cntr=0.3,0.1

Type RM Length L Ch R = 1 ,86719.4 ,287.7,303.1,355.6
XS GIS Cut Line= 2
     1745875.557      601232.912     1745360.639      601770.531
#Sta/Elev= 30
       0  762.89     9.8  761.24    19.6  758.62    39.2  752.68    58.8  746.43
   146.9  717.82   156.7  714.56   166.5  711.09   176.3  707.18   186.1  702.83
   215.5  689.06   264.5  666.56   274.3  662.64   284.1  659.86   293.8  658.21
   303.6  657.22   313.4   656.8     333  656.87   372.2  657.51   450.6  659.64
   568.1   662.3   577.9  662.89   587.7  664.45   597.5  667.36   617.1  674.16
   636.7  681.31   656.3  688.85   685.7  700.92   705.2  709.32   744.4   726.5
#Mann= 3 , 0 , 0
       0      .1       0   284.1    .045       0     333     .06       0
Bank Sta=284.1,333
XS Rating Curve= 0 ,0
Exp/Cntr=0.3,0.1

Type RM Length L Ch R = 1 ,86416.2 ,155.6,181.7,189.3
XS GIS Cut Line= 2
      1745710.41      601083.467     1745080.481      601448.398
#Sta/Elev= 30
       0  727.52    19.7  727.66    29.5  727.13    39.4  725.91      59  722.58
    68.9  720.39    88.5  714.88    98.4  711.51   108.2  707.62   147.6  689.86
   157.4  685.02   167.2  678.98   186.9  665.88   198.3  660.73   206.6  658.32
   216.4  656.78   226.3  656.46     246  656.67   354.2  656.87   393.5  657.68
   531.2  662.83   541.1  663.47   550.9  665.22   560.8  669.02     610  691.14
   629.6  700.49   649.3  710.58     669  719.71   708.3  735.82     728  743.01
#Mann= 3 , 0 , 0
       0      .1       0   198.3    .045       0     246     .06       0
Bank Sta=198.3,246
XS Rating Curve= 0 ,0
Exp/Cntr=0.3,0.1

Type RM Length L Ch R = 1 ,86234.6 ,119.5,101.7,102.4
XS GIS Cut Line= 3
     1745614.927      601071.315     1745441.041      601033.529
     1745079.301      601168.681
#Sta/Elev= 30
       0  707.88    18.7  702.88    37.5  698.09    46.8  695.82    65.6  691.58
    84.3  687.74    93.6  685.75     103  683.33   112.4  680.27   121.8  676.68
   140.5  669.08   149.8  665.52   159.2   662.4   168.4  659.96   177.9   658.1
   187.6  656.65   197.2  656.68   216.6   657.3   235.9  657.61   303.4  658.32
   380.7  659.44   448.3  660.86   467.6  661.34   477.2  661.83   486.9  663.25
   496.5  665.94   506.2  669.47   525.5  676.99   544.8  684.73   564.1  692.64
#Mann= 3 , 0 , 0
       0      .1       0   168.4    .045       0   216.6     .06       0
Bank Sta=168.4,216.6
XS Rating Curve= 0 ,0
Exp/Cntr=0.3,0.1

Type RM Length L Ch R = 1 ,86132.9 ,202.3,243,281.5
XS GIS Cut Line= 3
     1745635.833      600975.106      1745433.68      600931.177
     1745044.844      601076.453
#Sta/Elev= 30
       0  704.08     9.4  702.87    18.8  701.47    28.2  699.79      47     696
    75.2  690.66      94  687.37   103.4  685.93   112.8  684.68   131.6  682.52
   159.8  679.62   188.1  677.05   197.5  675.71   206.9  672.68   226.2  663.95
   235.8  661.04   245.5  659.71   255.1  658.74   264.8  657.61   274.4  656.75
   284.1  656.54   303.4  657.23   380.6  659.21   467.5  661.93   486.8  662.43
   496.5  662.78   506.1  663.73   515.8  665.76   525.4  668.84     622  704.38
#Mann= 3 , 0 , 0
       0     .08       0   264.8    .045       0   303.4     .08       0
Bank Sta=264.8,303.4
XS Rating Curve= 0 ,0
Exp/Cntr=0.3,0.1

Type RM Length L Ch R = 1 ,85889.9 ,355.2,356.5,355.8
XS GIS Cut Line= 2
      1745641.19      600967.123     1744983.162       600618.27
#Sta/Elev= 30
       0  703.08    29.4  698.02    68.6  690.24    88.2  686.76   117.6  682.62
     196  673.32   205.8  671.89   215.6  669.84   235.2  665.14     245  663.82
   333.2  659.81     398  657.56   421.4   656.7   431.2  656.89     441  658.94
   450.8  663.56     458  667.51   470.4  673.74   499.8  687.67   548.8  709.75
   568.4   719.2     588  730.05     637  758.12   656.6  768.49   676.2  778.13
   695.8  786.78   715.4   794.5   725.2  797.97     735     801   744.8  802.38
#Mann= 3 , 0 , 0
       0     .06       0     398    .045       0     458      .1       0
Bank Sta=398,458
XS Rating Curve= 0 ,0
Exp/Cntr=0.3,0.1

Type RM Length L Ch R = 1 ,85533.4 ,394.6,358.7,321.9
XS GIS Cut Line= 2
     1745912.788      600717.316     1745263.342      600367.312
#Sta/Elev= 30
       0  771.22    68.9  755.21   127.9  740.02   157.4  731.69   216.4  713.54
   245.9  704.08   275.4  694.89   285.3  691.56   295.1  687.47   304.9  682.77
   334.4  667.85   344.3  663.17   354.1  660.24     364  658.93   373.8  658.09
   393.5  656.98   432.8  655.85     469  655.32   491.8  655.01   501.7   655.1
   511.5  655.89   521.4  658.57     529  661.19     541  665.07   550.9  668.03
   570.5  673.54   609.9  683.12   629.6   688.2   698.4   708.4   737.8   719.4
#Mann= 3 , 0 , 0
       0     .06       0     469    .045       0     529      .1       0
Bank Sta=469,529
XS Rating Curve= 0 ,0
Exp/Cntr=0.3,0.1

Type RM Length L Ch R = 1 ,85174.7 ,620.3,582.9,544.7
XS GIS Cut Line= 2
     1746087.438      600028.668     1745308.392      600238.742
#Sta/Elev= 30
       0  774.66    39.4   763.4      59  756.99    88.6  746.52   118.1  733.86
   137.8  725.98   167.3  716.29   216.5  702.21     246  690.45   265.7  683.06
   285.4  676.27     305  670.36   324.7  666.03   354.2  662.77   403.4  659.34
   472.3  655.32     492  654.57   501.8  654.76   511.7  655.57   580.6  661.84
   590.4   664.2   610.1  672.86   619.9  676.62   629.8  679.39   639.6  681.48
   669.1  685.79   688.8  689.62   698.6  691.09   767.5  698.36   806.9  705.02
#Mann= 3 , 0 , 0
       0     .06       0   472.3    .045       0   511.7     .08       0
Bank Sta=472.3,511.7
XS Rating Curve= 0 ,0
Exp/Cntr=0.3,0.1

Type RM Length L Ch R = 1 ,84591.9 ,313.1,390.7,473.5
XS GIS Cut Line= 2
     1745344.627      599624.269     1744702.408      600948.025
#Sta/Elev= 30
       0  709.87      49  704.79    68.7  700.78   117.7  686.31   196.2  658.98
     206  656.64   229.1   654.5   264.8  652.71   289.1  653.88   441.4  663.68
   451.2  664.84     461  667.41   568.9  706.37   676.8  739.18   696.4  744.12
   765.1  758.87   814.1  773.11   843.6  780.25     873  784.93     922  789.69
   971.1  791.04   990.7  790.46  1039.7  787.01  1098.6     789    1128  787.42
  1157.4  783.91  1245.7  769.96  1363.4  753.86  1422.3  746.65  1471.3  741.76
#Mann= 3 , 0 , 0
       0     .08       0   229.1    .045       0   289.1     .06       0
Bank Sta=229.1,289.1
XS Rating Curve= 0 ,0
Exp/Cntr=0.3,0.1

Type RM Length L Ch R = 1 ,84201.2 ,444.4,448,436.4
XS GIS Cut Line= 3
     1745332.807      599630.067     1744578.139        599552.4
     1743917.501      600350.555
#Sta/Elev= 30
       0   707.8   116.7  695.92   155.6   693.5   233.4  676.42   291.8  656.39
   356.8  652.97     389  652.32   416.8     653   505.8  654.07   515.5  655.02
   525.2  657.98   671.1  738.09   758.6  780.96   807.5     794   846.6  799.17
     876  799.11  1012.8  790.38  1071.4     777  1120.3  768.44  1188.7  751.52
  1237.6  744.44  1296.2   741.7  1335.4  741.85  1364.7   744.2  1423.3  753.46
  1462.4  755.39  1569.9  739.74  1638.4  732.68  1745.9  728.73  1794.8   729.4
#Mann= 3 , 0 , 0
       0     .06       0   356.8    .045       0   416.8     .08       0
Bank Sta=356.8,416.8
XS Rating Curve= 0 ,0
Exp/Cntr=0.3,0.1

Type RM Length L Ch R = 1 ,83753.1 ,421.1,356.2,286.3
XS GIS Cut Line= 2
     1745486.783      599487.646     1744827.369       599146.05
#Sta/Elev= 30
       0  718.19    39.1  714.87    48.9  713.79    87.9  708.28    97.7  707.51
     127  706.76   146.6  705.53   166.1  703.74   185.7  700.17   234.5  690.32
   244.3  688.17   254.1  685.66   273.6  679.62   283.4  675.92   302.9  667.47
   312.7  664.32   322.5  662.62     342  660.96   381.1  658.46   491.7  652.51
   517.9  651.22   527.7  651.17   537.4  652.18   551.7  655.45   566.8  658.69
   605.8  665.29   635.2  671.24   664.5   677.8   723.1  691.49   742.6  695.52
#Mann= 3 , 0 , 0
       0     .06       0   491.7    .045       0   551.7      .1       0
Bank Sta=491.7,551.7
XS Rating Curve= 0 ,0
Exp/Cntr=0.3,0.1

Type RM Length L Ch R = 1 ,83396.9 ,542.3,538.8,532.7
XS GIS Cut Line= 3
     1745505.626       598569.05     1744982.239      599101.924
     1744785.923      599134.987
#Sta/Elev= 30
       0  779.33    29.5  773.87    88.4   766.3   117.9  761.14   167.1  748.18
   216.2  735.92   235.9  730.33   245.7  726.89   255.5  722.53   294.8  703.78
   314.5  695.02   334.2  685.13     344  679.08   363.6  664.87   373.5  659.66
   383.3  657.19   432.4  652.22   471.7  651.04   491.4  650.59   520.9  651.44
   609.3  655.32     629  658.19   638.8  660.48   678.1  672.05     688  673.52
   697.8   674.1   746.9  674.66   813.3  682.49   879.6  691.01     946   697.4
#Mann= 3 , 0 , 0
       0     .08       0   471.7    .045       0   520.9      .1       0
Bank Sta=471.7,520.9
XS Rating Curve= 0 ,0
Exp/Cntr=0.3,0.1

Type RM Length L Ch R = 1 ,82858.1 ,417.6,441.8,465.5
XS GIS Cut Line= 2
     1744888.277       598405.64      1744564.17      599067.434
#Sta/Elev= 30
       0  763.97      59  751.18    78.6  746.54    88.4  743.83   108.1  736.83
   147.4  724.06   157.2  721.18   176.9  716.14   186.7  713.04   196.5  709.46
   206.3  705.62   245.6  689.56   265.3  681.72   284.9  673.54   314.4  660.38
   324.2  656.73   334.1  654.35   353.7  650.92   363.5  649.85   373.4  649.75
     402  651.25   510.9   657.3   520.7  658.33   530.6  660.24   550.2  665.05
     560  667.84   579.7  673.84   599.3  680.06   658.3  699.38   736.9  726.05
#Mann= 3 , 0 , 0
       0     .08       0   353.7    .045       0     402      .1       0
Bank Sta=353.7,402
XS Rating Curve= 0 ,0
Exp/Cntr=0.3,0.1

Type RM Length L Ch R = 1 ,82416.3 ,376.7,406.4,433.9
XS GIS Cut Line= 2
     1744715.401       598305.87     1744060.815      598759.585
#Sta/Elev= 30
       0  732.26    19.7  726.35    98.3  700.35   157.3   681.4   196.7  669.07
   226.2  660.07     236  657.54   245.8  655.65   255.6  654.54   265.5  654.16
   421.5  651.29   442.5   649.8   452.3   649.4   462.1  650.73     472  654.99
   481.8  661.17   491.6   666.8   501.5  671.37   511.3  675.41   521.1  678.65
     531  680.96   540.8  682.42   550.6  684.65   560.5  687.72   570.3  690.17
   629.3  703.96   658.8  709.75   688.3  715.91   757.1  731.22   796.4  739.61
#Mann= 3 , 0 , 0
       0     .06       0   421.5    .045       0     472      .1       0
Bank Sta=421.5,472
XS Rating Curve= 0 ,0
Exp/Cntr=0.3,0.1

Type RM Length L Ch R = 1 ,82009.9 ,412.6,378.6,340.6
XS GIS Cut Line= 2
     1744704.539      598182.451     1743939.192      598162.259
#Sta/Elev= 30
       0  740.08    49.1  727.53    58.9  724.58    88.3  714.51    98.2  710.86
   127.6  698.54   147.2  689.79   166.9  680.68   215.9  657.02   225.8  652.63
   235.6  649.84   245.4  648.93   330.2  648.05   353.4  647.53   363.2   647.9
     373  649.77   390.2  655.26   422.1  665.75   441.7  673.02     481  689.63
     530  709.46   549.7  717.74   598.8   740.3   608.6  744.27   618.4  746.89
   628.2  748.12   667.5  748.99   726.4  751.92     746  752.29   765.6   751.7
#Mann= 3 , 0 , 0
       0     .06       0   330.2    .045       0   390.2      .1       0
Bank Sta=330.2,390.2
XS Rating Curve= 0 ,0
Exp/Cntr=0.3,0.1

Type RM Length L Ch R = 1 ,81631.3 ,500.6,457.3,416.3
XS GIS Cut Line= 3
     1748177.237      598247.108     1744404.187      597762.433
     1744085.314      598018.827
#Sta/Elev= 30
       0  920.31      59  908.13   176.9  866.12   363.7  809.32   530.8  853.59
   756.9  931.43   835.5  930.85   973.1  899.37  1277.8  793.58  1346.6  809.78
    1730  935.88  1867.6  934.09  2319.8  898.24  2526.2  809.04    2654  771.75
  2722.8  774.38  2811.3  763.06  2909.6  764.33  3007.9  746.37    3116  734.68
  3371.6  749.01  3499.3  743.27  3617.3  713.68  3735.2  655.45  3838.1  647.97
  3872.2  646.91  3898.1  648.14  3950.2  652.11  4028.1   679.9  4213.2  706.23
#Mann= 3 , 0 , 0
       0     .06       0  3838.1    .045       0  3898.1     .06       0
Bank Sta=3838.1,3898.1
XS Rating Curve= 0 ,0
Exp/Cntr=0.3,0.1

Type RM Length L Ch R = 1 ,81174.1 ,394.5,397.5,390.6
XS GIS Cut Line= 3
     1746509.626      594898.161      1743949.76      597436.109
     1744021.246      598080.652
#Sta/Elev= 30
       0  996.45   147.3  998.14   294.7  959.56   392.9  954.98   530.4  939.28
   677.7  940.18   805.4  918.17  1090.3  851.28  1375.1  703.57  1394.8  698.87
  1591.2  764.05  1758.2  724.88  1826.9  767.48  1974.2  833.13  2278.7  840.44
  2553.8  816.88  2858.2   799.8  3025.2  761.74  3221.7   726.5  3418.1  669.24
  3496.7  680.14  3604.7  711.67  3693.2  704.41  3819.5  650.46  3850.4  644.37
  3879.5  648.75  4046.9  654.47  4105.8  682.28  4174.6  697.42  4253.2  722.61
#Mann= 3 , 0 , 0
       0      .1       0  3819.5    .045       0  3879.5     .06       0
Bank Sta=3819.5,3879.5
XS Rating Curve= 0 ,0
Exp/Cntr=0.3,0.1

Type RM Length L Ch R = 1 ,80776.5 ,375.9,376.5,387
XS GIS Cut Line= 2
     1743550.098      597488.384     1743754.099      598190.681
#Sta/Elev= 30
       0  728.34    29.2  718.57    58.5   709.4    97.5   697.7   165.8  678.06
     234  657.22   243.8   654.5   253.5  652.64   263.3  651.85   341.3  650.09
     351  649.61   362.4  647.59   370.5  645.68   380.3  644.29     390  644.21
   399.8  645.28   409.5  646.74   419.3  647.72   422.4  647.87   497.3  650.56
     507  651.17   516.8  653.84   526.6  658.62   575.3  684.91   585.1   689.6
   594.8  693.49   633.8  707.03   663.1  717.47   702.1  731.73   731.3  742.64
#Mann= 3 , 0 , 0
       0     .06       0   362.4    .045       0   422.4     .06       0
Bank Sta=362.4,422.4
XS Rating Curve= 0 ,0
Exp/Cntr=0.3,0.1

Type RM Length L Ch R = 1 ,80400.1 ,306.6,309,311.3
XS GIS Cut Line= 3
     1743304.132      597560.479     1743306.716       597618.92
     1743340.357      598379.744
#Sta/Elev= 30
       0  711.16      39   697.5      78  685.08   126.8  670.75   165.9  658.82
   175.7  656.01   185.4   654.1   195.2  653.22   292.8  649.19   351.4  647.87
   419.8  647.76   429.5   647.1   433.2  646.48     449  643.89   458.8  643.53
   468.6  644.57   488.1  648.31   493.2   649.6   497.9  650.79   517.4  658.39
   546.7   671.1   595.5  692.98   624.8  705.57   654.1  717.06   693.1  731.28
   722.4   741.1   751.7  749.82   761.5  752.05   790.8     757   820.1  763.73
#Mann= 3 , 0 , 0
       0     .06       0   433.2    .045       0   493.2     .08       0
Bank Sta=433.2,493.2
XS Rating Curve= 0 ,0
Exp/Cntr=0.3,0.1

Type RM Length L Ch R = 1 ,80091   ,442.3,448.3,450.8
XS GIS Cut Line= 2
     1743040.095      597556.023     1743036.337      598621.348
#Sta/Elev= 30
       0  742.45    39.1  722.17    68.4   710.1      88  704.38   136.8  693.24
   166.2  684.76   175.9  680.44   224.8  653.76   234.6  649.49   244.3  646.97
   254.1  646.09   336.4  645.66   361.6   645.3     391  643.08   400.7  643.51
   478.9  651.16   488.7  654.93   537.6  678.81   547.3  682.05   557.1  683.88
   703.7  698.18   742.8  703.41   752.6  703.87   811.2  699.13   869.9  691.98
   879.6  692.43   889.4  695.18   928.5  710.46     948  715.58  1065.3  735.73
#Mann= 3 , 0 , 0
       0     .08       0   336.4    .045       0   400.7     .06       0
Bank Sta=336.4,400.7
XS Rating Curve= 0 ,0
Exp/Cntr=0.3,0.1

Type RM Length L Ch R = 1 ,79642.8 ,304.9,345.2,385.5
XS GIS Cut Line= 2
      1742669.37      597658.809     1742631.673      598431.744
#Sta/Elev= 30
       0  696.33    58.8  690.88   107.8  687.36   117.6  685.52   127.3  681.71
   137.1  676.64   156.7  665.53   166.5   659.2   170.5  656.15   176.3  651.72
   186.1  645.46   195.9  643.08   205.7  643.23   230.5  645.88   244.9  647.37
   293.9  651.86   342.8  656.99   460.4  671.41   519.2  677.95     529  679.64
   558.4  685.93   587.7  691.66   607.3  696.07   617.1  698.56   636.7  703.97
   646.5  706.87   685.7  719.07   715.1  727.92   754.3  739.31   773.8  744.66
#Mann= 3 , 0 , 0
       0      .1       0   170.5    .045       0   230.5     .06       0
Bank Sta=170.5,230.5
XS Rating Curve= 0 ,0
Exp/Cntr=0.3,0.1

Type RM Length L Ch R = 1 ,79297.6 ,427.9,468.9,509.9
XS GIS Cut Line= 2
     1742772.117      597518.129     1742005.996      598112.348
#Sta/Elev= 30
       0  725.85    29.4  720.63    78.4  709.52    97.9  705.84   166.5  694.28
   244.8  679.85     284  673.36   313.4  669.58   362.4  665.58   470.1  654.57
   528.8  649.44   537.6  647.63   548.4  644.43   558.2  642.82     568  643.07
   577.8  644.65   597.6  649.12   636.6  660.82   646.4  663.61   656.2  665.89
     666  667.39   734.5  675.68   744.3  677.58   754.1  680.06   763.9  683.54
   773.7  688.19   832.4  720.11   871.6  740.21   920.6  763.82   969.6  786.22
#Mann= 3 , 0 , 0
       0     .08       0   537.6    .045       0   597.6      .1       0
Bank Sta=537.6,597.6
XS Rating Curve= 0 ,0
Exp/Cntr=0.3,0.1

Type RM Length L Ch R = 1 ,78828.7 ,308.3,299.7,289.7
XS GIS Cut Line= 2
     1742667.088      597562.814     1741921.099      597357.166
#Sta/Elev= 30
       0  698.85    39.2  690.32    78.4  681.18   146.9  667.64   156.7  666.17
   186.1  663.49   205.7  661.46   225.3  659.12   274.3  652.75   293.8  650.45
   323.2  647.43   333.8  645.95   342.8  644.34   352.6  642.95   362.4   642.8
   372.2   644.7     382  649.33   391.8  655.23   411.4  666.89   440.8  684.73
   450.6  690.01   460.4  694.16   499.6  707.62   538.7   720.5   617.1  745.25
   675.9  764.47   685.7   767.2   695.4  768.28   705.2   767.4   773.8  757.29
#Mann= 3 , 0 , 0
       0     .06       0   333.8    .045       0   391.8      .1       0
Bank Sta=333.8,391.8
XS Rating Curve= 0 ,0
Exp/Cntr=0.3,0.1

Type RM Length L Ch R = 1 ,78529   ,313.5,305.7,299.2
XS GIS Cut Line= 2
      1742784.05      597226.118     1742012.578      597165.944
#Sta/Elev= 30
       0  740.43    19.6  735.06      49  725.68    88.2  714.11      98  710.56
   117.5  702.43   176.3  672.66   186.1  668.53   195.9  665.38   205.7  663.18
   244.9  658.09   313.4  645.29     333  642.71   342.8  642.71   352.6  643.92
   360.6  645.84   372.2  648.08     431  653.62   489.8  664.82   499.6  666.29
   519.1   668.1   528.9  670.15   548.5  677.77   626.9  711.79   695.4  742.66
   705.2  746.44     715  748.63   724.8  748.94   754.2   747.4   773.8   745.7
#Mann= 3 , 0 , 0
       0     .06       0   313.4    .045       0   360.6     .06       0
Bank Sta=313.4,360.6
XS Rating Curve= 0 ,0
Exp/Cntr=0.3,0.1

Type RM Length L Ch R = 1 ,78223.3 ,360.2,352.8,345.4
XS GIS Cut Line= 2
     1742705.767       596875.26     1741977.985      596947.045
#Sta/Elev= 30
       0  759.74    48.8  744.15    58.5  739.78   214.5   655.7   224.3  649.93
     234  645.02   243.8  642.96   253.5  643.56     273  648.34   280.3  649.12
   341.3  650.66   370.5  652.24   458.3  662.14     468   664.5   477.8  668.29
   516.8  687.17   526.6  691.01   536.3  693.25     546  694.16     585  695.72
   594.8  695.32   604.6  694.04   614.3  691.71   633.8  685.44   653.3  678.33
   672.8     670   682.6  667.51   692.3   667.3   702.1  668.85   731.3  677.13
#Mann= 3 , 0 , 0
       0      .1       0   224.3    .045       0   280.3     .06       0
Bank Sta=224.3,280.3
XS Rating Curve= 0 ,0
Exp/Cntr=0.3,0.1

Type RM Length L Ch R = 1 ,77870.5 ,388.1,360,331.9
XS GIS Cut Line= 2
     1742967.063      596398.456     1741911.073      596680.307
#Sta/Elev= 30
       0  809.61    29.3  811.76    58.6  813.24   146.4   814.2   175.6     815
   185.4  814.86   195.2  813.69   204.9  811.26     283  787.33   400.1   748.1
   409.9  743.72   458.6  719.65   585.5   658.4     605  647.47   614.8  643.52
   624.6  642.66   655.1  646.38   722.1  647.12   790.4  650.78   800.2  651.67
     810   654.3   819.7   658.9   878.3  689.53   897.8  699.05   907.5  702.97
   917.3  705.84   966.1   717.2   975.8  718.86  1044.2  723.67    1093  725.86
#Mann= 3 , 0 , 0
       0      .1       0     605    .045       0   655.1     .06       0
Bank Sta=605,655.1
XS Rating Curve= 0 ,0
Exp/Cntr=0.3,0.1

Type RM Length L Ch R = 1 ,77510.5 ,358.6,326.8,294.9
XS GIS Cut Line= 2
     1742508.638      595870.481     1741943.398      596551.826
#Sta/Elev= 30
       0  679.48    49.2  695.18    68.9  700.08    88.5   703.3   127.9  707.61
   147.6  709.23   255.8  713.36   265.6  712.84   275.4  710.91   344.3  688.53
   462.3   652.2     476  647.07     482  644.65   491.8  642.75   501.7  642.37
   511.5  642.51     536  645.25   550.8  646.57     600   645.8   649.2  645.84
     659  646.33   668.9   649.1   688.6  658.32   708.2  668.86   747.6  690.82
   757.4  695.67   767.2  699.43   816.4  713.87   855.8  723.06   885.3  728.45
#Mann= 3 , 0 , 0
       0      .1       0     476    .045       0     536      .1       0
Bank Sta=476,536
XS Rating Curve= 0 ,0
Exp/Cntr=0.3,0.1

Type RM Length L Ch R = 1 ,77183.7 ,391.4,373.1,354.9
XS GIS Cut Line= 2
     1741887.175       595783.25     1741897.159      596536.389
#Sta/Elev= 30
       0  803.94    19.6  792.53    29.4  787.23    58.7  771.87      88  756.68
    97.8  751.83   107.6  747.13   117.4  742.68   176.1  716.86   244.6  686.52
   283.7  668.88     313  655.51     325   649.4   332.6  645.43   342.4  642.49
   352.2  642.35   371.7  644.72   381.5  645.33     385  645.44   498.9   649.4
   508.7  650.02   518.4  651.49   528.2   653.9   557.6  662.23   567.4  665.26
   655.4  694.13     675  700.79   694.5  707.72   723.9  718.63   753.2  729.65
#Mann= 3 , 0 , 0
       0      .1       0     325    .045       0     385      .1       0
Bank Sta=325,385
XS Rating Curve= 0 ,0
Exp/Cntr=0.3,0.1

Type RM Length L Ch R = 1 ,76810.6 ,378.6,375.1,371.6
XS GIS Cut Line= 2
     1741397.742      595932.797     1741691.973      596598.689
#Sta/Elev= 30
       0  757.25    39.4  753.13    68.9  750.33    78.7  749.51   137.7  745.31
   147.6     744   157.4   741.1   167.2  737.07   177.1  732.35   196.8  722.41
   226.3  707.31   314.8  660.86   324.6  655.36     334  649.41   344.3  644.18
   354.2  642.33     364  642.38     394  644.28   432.9  646.56     482  649.75
   531.2  652.77   541.1  653.98   550.9  656.63   560.8  660.31   590.3  672.46
   629.6  688.87   659.1  700.97   678.8  708.86   708.3  720.42     728  727.86
#Mann= 3 , 0 , 0
       0      .1       0     334    .045       0     394      .1       0
Bank Sta=334,394
XS Rating Curve= 0 ,0
Exp/Cntr=0.3,0.1

Type RM Length L Ch R = 1 ,76435.5 ,443.5,453.8,463.9
XS GIS Cut Line= 2
     1741035.853      596105.764     1741380.835      596747.512
#Sta/Elev= 30
       0  688.87    38.9  677.89    58.3  674.21    77.7  672.43   126.3  671.87
   165.2  669.12   242.9  659.38   252.6  658.65     272  658.34   281.7  657.63
   301.2  654.47   312.3  651.21   330.3  643.75     340  641.38   349.7  641.09
   372.3  644.04   388.6  645.32   485.7  649.12   495.4  649.64   505.2  651.02
   514.9  653.69   553.7   666.7   573.2  673.64   592.6  681.25   621.7  694.36
   660.6  713.97   689.7  727.64   709.2  735.63   718.9  738.85   728.6  741.53
#Mann= 3 , 0 , 0
       0      .1       0   312.3    .045       0   372.3      .1       0
Bank Sta=312.3,372.3
XS Rating Curve= 0 ,0
Exp/Cntr=0.3,0.1

Type RM Length L Ch R = 1 ,75981.6 ,354.1,350.2,346.3
XS GIS Cut Line= 2
     1740719.198      596270.254     1740911.638      596973.241
#Sta/Elev= 30
       0  704.21    19.4  700.76    58.3  692.97   145.8  676.82   184.6  668.76
   213.8  661.98   233.2  658.27   252.7  655.36   334.2  647.25   340.1  646.54
   349.8  644.03   359.6  640.54   369.3  638.83     379  639.17   394.2  642.31
   398.4  643.26   408.2   644.9   427.6   647.5   437.3  649.71     447  653.73
   456.8  658.93   476.2  670.13   524.8  699.52   534.5  705.04   544.2  709.84
   612.2  738.21   670.5  765.17     690  773.75   709.4  781.68   728.8   788.7
#Mann= 3 , 0 , 0
       0      .1       0   334.2    .045       0   394.2      .1       0
Bank Sta=334.2,394.2
XS Rating Curve= 0 ,0
Exp/Cntr=0.3,0.1

Type RM Length L Ch R = 1 ,75631.4 ,378.3,375.9,372.3
XS GIS Cut Line= 2
     1740350.633      596369.143     1740603.465      597052.883
#Sta/Elev= 30
       0  727.73    38.9   719.4    58.3  715.57   106.9  707.39   126.4  703.68
   145.8  699.31   223.6  681.06     243   676.1   262.4  670.67   272.2  667.48
   291.6  660.53     335  645.59   349.9  640.59   359.6  638.89   369.4  639.15
   379.1  641.23   388.8  643.56     395  644.41   398.5  644.89   408.2  645.69
   447.1  648.51     486  651.86   495.7  653.34   505.4  656.06   544.3  669.77
   563.8  676.98   612.4  695.65   699.8  730.04   719.3  737.08     729  739.53
#Mann= 3 , 0 , 0
       0      .1       0     335    .045       0     395      .1       0
Bank Sta=335,395
XS Rating Curve= 0 ,0
Exp/Cntr=0.3,0.1

Type RM Length L Ch R = 1 ,75255.5 ,380.4,357.3,335.2
XS GIS Cut Line= 2
     1739972.497      596460.478     1740278.702      597145.328
#Sta/Elev= 30
       0  768.33    77.9  744.36   155.9  721.68   194.8  709.87   233.8  697.24
     302  673.79   331.2  664.08   370.2     652   395.3  644.92   409.2  641.56
   418.9  639.57   428.7  638.54   438.4  638.64   448.2  640.09   455.3  641.61
   467.6  643.92   477.4  644.99   565.1  650.72     604  653.93   613.8  655.72
   623.5  658.48   652.8  667.88   672.2  673.58     682  675.85   691.7  677.48
   701.5  677.99   711.2  677.27   730.7  674.44   740.4  674.13   750.2  675.66
#Mann= 3 , 0 , 0
       0      .1       0   395.3    .045       0   455.3      .1       0
Bank Sta=395.3,455.3
XS Rating Curve= 0 ,0
Exp/Cntr=0.3,0.1

Type RM Length L Ch R = 1 ,74898.3 ,470.3,413.9,357.3
XS GIS Cut Line= 2
     1739512.121      596787.544     1740181.899      597276.402
#Sta/Elev= 30
       0  737.15    97.6  734.58   146.3  736.04   156.1  736.09   175.6  735.12
   185.4  735.13   214.6  738.03   224.4  737.58   234.1  735.56   253.6  729.98
   263.4   726.4   273.2   722.3   292.7  713.11   321.9  696.97   394.2  653.13
   409.7  642.44   419.5  639.04   429.2  638.88   448.8  642.66   454.2  643.33
     478     645   624.3  652.95   653.6  656.74   712.1  665.73   721.9  666.65
   741.4  667.22   751.2  667.94   760.9   669.2   809.7  677.31   829.2  680.05
#Mann= 3 , 0 , 0
       0      .1       0   394.2    .045       0   454.2      .1       0
Bank Sta=394.2,454.2
XS Rating Curve= 0 ,0
Exp/Cntr=0.3,0.1

Type RM Length L Ch R = 1 ,74484.4 ,289.3,278,266.5
XS GIS Cut Line= 2
      1739676.64       597537.22     1740096.113      597244.769
#Sta/Elev= 30
       0  684.47    29.5  694.47    39.3  697.48    49.2  699.64      59  700.97
    68.8  702.58    88.5  706.41    98.3  707.94   108.2  707.46     118  703.24
   137.7  690.76   157.3  677.97   167.2  671.61   186.8  659.26   197.7  652.12
   206.5  645.85   216.3  639.97   226.2  638.14     236  639.61   245.8  642.43
   255.7  644.54   257.7  644.72   265.5  645.44   393.4  651.29   442.5  653.82
   452.4  654.56   462.2  655.54     472  656.73   491.7  659.45   511.4  662.66
#Mann= 3 , 0 , 0
       0      .1       0   197.7    .045       0   257.7      .1       0
Bank Sta=197.7,257.7
XS Rating Curve= 0 ,0
Exp/Cntr=0.3,0.1

Type RM Length L Ch R = 1 ,74206.4 ,202.2,222.4,242.5
XS GIS Cut Line= 2
      1739908.79      597774.889     1740294.181       597326.39
#Sta/Elev= 30
       0  701.28    38.8  703.31    77.6  705.68    87.2  705.44    96.9  703.39
   116.3  695.58   155.1  679.03   184.2  667.35   203.6  660.04     223  653.25
   232.7  650.12   250.3  644.98   261.7  641.21   271.4  638.45   281.1  637.36
   290.8  638.28   300.5   640.6   310.3  643.28   319.9   645.4   368.4  651.83
   378.1  653.48   407.2  660.41   426.5  664.51   436.2  666.24   455.6  669.16
     475  672.72   504.1  679.74   552.6   692.6     572  697.13   591.3  701.11
#Mann= 3 , 0 , 0
       0      .1       0   250.3    .045       0   310.3      .1       0
Bank Sta=250.3,310.3
XS Rating Curve= 0 ,0
Exp/Cntr=0.3,0.1

Type RM Length L Ch R = 1 ,73984   ,289.5,325.4,361.3
XS GIS Cut Line= 2
      1740032.62       597808.36     1740557.419      597575.247
#Sta/Elev= 30
       0  692.71    38.9  682.85    68.1  675.83   116.8  664.73   155.7  656.52
   215.9     645   223.9  643.16   233.6  640.17   243.3  637.69   253.1  637.38
   262.8  638.91   275.9  643.26     292  648.59   301.7   652.1   311.4  656.71
   321.2     662   340.6  672.96   360.1  684.47   379.6  696.44   418.5  720.92
     438  732.62   457.4  743.29   467.2  748.17   476.9  752.68   486.6  756.89
   496.4  760.72   515.8  767.41   525.6  770.28     545  774.96   574.2  780.31
#Mann= 3 , 0 , 0
       0      .1       0   215.9    .045       0   275.9      .1       0
Bank Sta=215.9,275.9
XS Rating Curve= 0 ,0
Exp/Cntr=0.3,0.1

Type RM Length L Ch R = 1 ,73658.6 ,197.7,197.6,197.8
XS GIS Cut Line= 2
      1740013.48      597905.283     1740627.849       598149.09
#Sta/Elev= 30
       0  695.15    19.4  690.11    38.9  685.49    97.2  672.68   145.8  662.95
   233.3  646.32     243   643.8     254  639.86   262.4  637.28   272.2  636.45
   281.9  637.49     311  644.85     314  645.89   320.8  648.26   330.5  653.23
   379.1  682.67   398.5  693.31     418  702.85   476.3  729.88     486  734.17
   495.7  737.92   505.4  741.31   524.9  747.37   534.6  750.82     554   758.8
   583.2  771.85   612.4  786.36   631.8   795.3   641.5  798.57     661   803.4
#Mann= 3 , 0 , 0
       0      .1       0     254    .045       0     314      .1       0
Bank Sta=254,314
XS Rating Curve= 0 ,0
Exp/Cntr=0.3,0.1

Type RM Length L Ch R = 1 ,73461   ,292.4,289.8,286.9
XS GIS Cut Line= 3
     1739905.378      598073.374     1740582.046      598341.904
     1740583.617      598342.527
#Sta/Elev= 30
       0  694.29    49.2   693.7      59  693.09    68.9  691.33   186.9  662.38
   255.8  646.08   268.4  642.07   275.5  639.52   285.3  636.98   295.1  636.41
     305  637.65   314.8  640.31   324.6  642.59   328.4  643.13   334.5     644
   344.3  644.91   354.2  646.56     364  650.15   442.7  689.96   482.1  711.19
   511.6  728.26   521.4  733.69   531.2  738.09   541.1  741.46   629.6  768.54
   639.5   771.3   659.1  776.16   688.6  782.49   708.3   786.5   729.7  790.23
#Mann= 3 , 0 , 0
       0      .1       0   268.4    .045       0   328.4      .1       0
Bank Sta=268.4,328.4
XS Rating Curve= 0 ,0
Exp/Cntr=0.3,0.1

Type RM Length L Ch R = 1 ,73171.1 ,273.8,296.4,319.1
XS GIS Cut Line= 3
     1739814.754      598362.974     1740506.634      598589.446
     1740525.727      598595.696
#Sta/Elev= 30
       0  682.64    68.9  679.94    78.7  679.37    88.5  677.88   196.8  649.41
   206.6  646.58   212.5  644.12   226.3  637.96   236.1  636.32     246   636.2
   255.8  636.48   272.5  638.45   334.5  643.74   354.2  647.06     364  650.06
   373.8  654.48   383.7  660.08   403.4  672.37   413.2  677.89     423  682.58
   432.9   686.2   452.5  692.21   462.4  695.09   472.2  697.19   491.9   700.2
   560.8  708.59     610  712.96   649.3  717.26   718.2  725.84   748.1  730.96
#Mann= 3 , 0 , 0
       0      .1       0   212.5    .045       0   272.5      .1       0
Bank Sta=212.5,272.5
XS Rating Curve= 0 ,0
Exp/Cntr=0.3,0.1

Type RM Length L Ch R = 1 ,72874.7 ,173.6,220.3,266.9
XS GIS Cut Line= 2
     1739765.923      598563.302     1740938.822      599815.423
#Sta/Elev= 30
       0   666.9    78.4  661.47      98   656.1   130.4  643.88   147.1  638.34
   166.7  636.09   190.4  641.93   313.7  645.66   382.4  662.84   421.6  675.24
   480.4  701.34   607.8  748.03   656.8  771.33   676.5  779.16   705.9  787.36
   774.5     799   852.9  822.25   921.6  838.97  1019.6  853.37    1049  859.08
  1078.4  868.76  1107.8  882.59  1176.4  897.11  1225.5  917.89  1294.1  936.01
  1392.1  949.46    1451  952.73  1666.6  954.26  1686.2  951.86  1715.7  945.71
#Mann= 3 , 0 , 0
       0      .1       0   130.4    .045       0   190.4     .08       0
Bank Sta=130.4,190.4
XS Rating Curve= 0 ,0
Exp/Cntr=0.3,0.1

Type RM Length L Ch R = 1 ,72654.4 ,234.6,291.9,349.2
XS GIS Cut Line= 2
     1739798.508      598381.285     1739364.057      600041.028
#Sta/Elev= 30
       0  681.49    39.2  679.16   196.1  664.63   254.9  663.18   323.5  657.29
   343.1  653.62   393.4  640.38   411.8  636.45   421.6  635.81   453.4  639.73
   470.6  641.21   578.4  642.13   607.8  646.99   666.7  675.44   725.5  708.52
   803.9  749.79   862.7  778.63   892.1  791.74   911.8  796.92  1029.4  819.42
  1137.2  827.19  1225.5  837.48  1254.9  838.95  1313.7  836.77  1333.3   834.8
  1539.2  792.76  1568.6  788.28    1647  779.87  1666.6  780.16  1715.7  796.56
#Mann= 3 , 0 , 0
       0      .1       0   393.4    .045       0   453.4     .08       0
Bank Sta=393.4,453.4
XS Rating Curve= 0 ,0
Exp/Cntr=0.3,0.1

Type RM Length L Ch R = 1 ,72362.5 ,325.7,324.5,323.3
XS GIS Cut Line= 3
      1739766.58      598386.275     1739713.615      598664.222
     1739236.881      598698.821
#Sta/Elev= 30
       0  676.85    29.3  675.06    97.6  668.24   117.1  668.09   126.8  667.11
   146.4  662.93   185.4  658.93   214.6  658.02   224.4  658.66   243.9  660.83
   253.7  661.21   263.4  660.97   302.5   657.5   312.2  656.06   341.5  649.68
     361  647.25     400  646.47   487.8   643.2     499   641.6   517.1  636.62
   526.8  635.71   536.6  636.33     559  640.41   575.6  641.04   585.4  643.22
   614.6  661.44   634.1  672.06   663.4     687   702.4  710.78   760.9  742.95
#Mann= 3 , 0 , 0
       0     .08       0     499    .045       0     559      .1       0
Bank Sta=499,559
XS Rating Curve= 0 ,0
Exp/Cntr=0.3,0.1

Type RM Length L Ch R = 1 ,72038.1 ,455.5,455.7,455.4
XS GIS Cut Line= 2
     1739792.113      598335.264      1739209.44      598392.307
#Sta/Elev= 30
       0  684.48     9.8   682.2    29.3  674.33    68.3  657.86    87.8  649.82
    97.6  646.98   107.3  645.79   117.1  645.39   146.4  644.65   195.2  643.91
   224.4  642.98   234.2  642.27   243.9  640.72   245.9  640.22   253.7  638.25
   263.5  636.24   273.2  635.67     283  636.36   305.9  640.45   312.2  641.46
     322  642.52   331.8   644.1   341.5  647.12   380.6  662.07   419.6  676.66
   439.1  684.35   478.1  700.22   517.2  715.74   536.7  723.74   585.5  744.59
#Mann= 3 , 0 , 0
       0     .08       0   245.9    .045       0   305.9     .08       0
Bank Sta=245.9,305.9
XS Rating Curve= 0 ,0
Exp/Cntr=0.3,0.1

Type RM Length L Ch R = 1 ,71582.4 ,463.9,454.5,445.1
XS GIS Cut Line= 2
     1739870.298      597909.797     1739287.626       597966.84
#Sta/Elev= 30
       0   698.4    58.6  697.82    68.3  697.33    78.1  695.84    87.8  691.68
    97.6  685.24   107.3  678.62   126.8   665.8   136.6  659.66   146.4  653.77
   156.1   648.2   165.9  644.34   175.6   642.5   185.4  641.46   196.4  639.98
   214.7  636.16   224.4  635.31   234.2  635.32   256.4  636.77   273.2   637.9
   292.7  639.55   302.5  640.18   380.6  641.95   409.8  642.29   419.6  643.06
   429.3  645.21   487.9  663.86   546.4  682.77   556.2  686.02   585.5  696.16
#Mann= 3 , 0 , 0
       0      .1       0   196.4    .045       0   256.4     .08       0
Bank Sta=196.4,256.4
XS Rating Curve= 0 ,0
Exp/Cntr=0.3,0.1

Type RM Length L Ch R = 1 ,71127.9 ,433.6,420.6,413.5
XS GIS Cut Line= 2
      1739701.43      597448.807      1738767.59      597744.602
#Sta/Elev= 30
       0  701.95     9.8  700.02    19.6  696.91    58.8   682.8    88.2   670.9
   107.8  661.55   137.1  641.68   146.9  637.44   156.7  635.38   172.4  634.64
   176.3   634.6   195.9  635.04   232.4  638.54   342.8  639.21   352.6   640.2
   362.4  642.52   391.8  652.96   470.2  682.89   519.2  700.17   607.3   728.7
   666.1  745.37   675.9  745.62   685.7   743.7   852.2  700.79     862   698.4
   871.8  697.61   881.6  698.54   891.4  701.03   940.4  718.35   979.6  731.27
#Mann= 3 , 0 , 0
       0      .1       0   172.4    .045       0   232.4     .08       0
Bank Sta=172.4,232.4
XS Rating Curve= 0 ,0
Exp/Cntr=0.3,0.1

Type RM Length L Ch R = 1 ,70707.2 ,454.3,416.8,371.3
XS GIS Cut Line= 2
      1739682.68      597028.337      1739128.06       597215.84
#Sta/Elev= 30
       0  719.32    29.3  715.53      39     713    78.1  700.63    87.8  697.38
    97.6  693.69   107.3  689.07   185.4  646.65   195.2  642.77   204.9  641.48
   214.7  640.89   234.2  638.96   263.5  634.48   273.2   633.6     283  633.38
   293.6  633.84   302.5  634.99     322  639.42   331.8  640.41   341.5  640.58
   439.1  640.89   448.8  641.04   458.6  642.14   468.4  645.16   487.9  654.15
   526.9  672.88   536.7  676.55   546.4  678.32   556.2  678.77   585.5  679.27
#Mann= 3 , 0 , 0
       0      .1       0   293.6    .045       0   341.5     .08       0
Bank Sta=293.6,341.5
XS Rating Curve= 0 ,0
Exp/Cntr=0.3,0.1

Type RM Length L Ch R = 1 ,70290.5 ,340,335.5,330.3
XS GIS Cut Line= 2
     1739211.186      596610.551      1739050.19      597280.314
#Sta/Elev= 30
       0  716.64    29.5   705.8    39.4  704.36    49.2  705.33    78.7  713.16
    88.6  714.26    98.4  711.69   118.1  699.84   167.3  663.42     187  651.13
   196.8  646.37   206.6  642.63   216.5  639.81   236.2  636.38   252.2  636.29
   265.7  635.88   285.4   633.5   295.2  633.68   312.2  637.54   324.7  640.49
   383.8  646.16   403.5   649.1   472.4  666.61     492  670.18   541.2  674.57
   570.8  678.81   600.3  678.38   629.8  678.89   659.3  678.21   688.8  680.02
#Mann= 3 , 0 , 0
       0      .1       0   252.2    .045       0   312.2     .08       0
Bank Sta=252.2,312.2
XS Rating Curve= 0 ,0
Exp/Cntr=0.3,0.1

Type RM Length L Ch R = 1 ,69955   ,258.9,275.6,292.1
XS GIS Cut Line= 2
     1738871.732      596645.822     1738786.344      597254.109
#Sta/Elev= 30
       0  705.32     9.8  708.74    19.5  711.01    29.2  711.07      39  710.37
    48.8  709.22    58.5  707.22    68.2  704.13      78     700    87.8  695.34
   107.2  684.96   146.2  662.66   165.8  652.61   182.3  644.88     195  638.61
   204.8  634.96   214.5  633.43   224.2  633.71   242.3  636.76   253.5  638.46
   292.5  643.01   370.5  651.27   409.5  655.96   419.2   657.4     429  659.72
   458.2  668.96   497.2  680.62   575.2  702.73   604.5  710.45   614.2  712.16
#Mann= 3 , 0 , 0
       0      .1       0   182.3    .045       0   242.3     .08       0
Bank Sta=182.3,242.3
XS Rating Curve= 0 ,0
Exp/Cntr=0.3,0.1

Type RM Length L Ch R = 1 ,69679.3 ,420.9,469.3,517.8
XS GIS Cut Line= 2
      1738716.08      596562.725     1738370.984      597177.113
#Sta/Elev= 30
       0  683.32    19.6   683.3    39.2  682.57    78.3  679.54    88.1  678.28
    97.9  676.44     137  668.14   244.7  643.88   254.5  641.19   257.2  640.11
     274  633.57   283.8  631.96   293.6  632.39   303.4  634.56   317.2  638.13
     323  639.43   362.1   646.8   411.1  656.41   420.8   658.7   430.6  661.79
   450.2  669.17   479.6  680.93   538.3  705.09   557.9  712.72   577.4  719.89
   606.8  730.02   665.5  749.08   675.3  751.76   694.9  756.22   704.7  758.74
#Mann= 3 , 0 , 0
       0      .1       0   257.2    .045       0   317.2      .1       0
Bank Sta=257.2,317.2
XS Rating Curve= 0 ,0
Exp/Cntr=0.3,0.1

Type RM Length L Ch R = 1 ,69210   ,345.9,395.1,443.8
XS GIS Cut Line= 2
     1738662.434       596501.26     1737962.684      596491.942
#Sta/Elev= 30
       0   672.5    58.3  669.08      68  668.13    77.8  666.81    97.2  663.75
     175  650.17   184.7  648.73   194.4  647.84   204.1  647.29   301.3  642.22
     311  641.32   320.8  639.51   322.9   638.9   340.2  633.59   349.9  631.72
   359.6  632.36   369.3  636.01   382.9  643.59   388.8  646.78   417.9  660.62
   495.7  697.06     554   723.6   563.7  727.83   573.5   731.2   583.2  732.09
   592.9   730.8   612.3  727.47   660.9  718.34   680.4  714.52   699.8  710.36
#Mann= 3 , 0 , 0
       0      .1       0   322.9    .045       0   382.9      .1       0
Bank Sta=322.9,382.9
XS Rating Curve= 0 ,0
Exp/Cntr=0.3,0.1

Type RM Length L Ch R = 1 ,68814.9 ,418.2,411.1,404.3
XS GIS Cut Line= 2
     1738715.643      596485.071     1738418.605      595918.375
#Sta/Elev= 30
       0  667.82    38.8  661.72    77.6  656.34   106.6  651.16     126  648.63
   174.5  645.16   271.4  639.17     282  638.09   290.8  636.35   310.2  631.64
   319.9  632.52   329.6  637.91     342  649.07     349  654.96   358.7  662.21
   378.1  675.57   397.5  687.34   407.2  692.74   426.6  702.66   445.9  711.49
     475  722.98   494.4  729.66   513.8  735.32   523.5  737.72   533.2  738.61
   542.9  737.61   562.3  734.35     601  729.18   620.4  725.69   639.8  720.77
#Mann= 3 , 0 , 0
       0      .1       0     282    .045       0     342      .1       0
Bank Sta=282,342
XS Rating Curve= 0 ,0
Exp/Cntr=0.3,0.1

Type RM Length L Ch R = 1 ,68403.8 ,403,368.5,332.8
XS GIS Cut Line= 2
     1739138.674       596311.27     1738796.096      595845.196
#Sta/Elev= 30
       0  700.74    19.6  692.48      49  680.45    88.2  664.96      98   661.3
   107.8  657.92   117.6  654.87   137.3  648.29   147.1  645.25   156.9  643.69
   166.7   643.1   205.9   641.2   264.7  638.86   274.5  638.36   285.4  637.13
   294.1  635.26   303.9  632.47   313.7  631.51   323.5  632.92   333.3  636.86
   343.1  641.95   345.4     643     402  668.19   431.4  681.59   460.8  695.27
   470.6  699.64   480.4  702.94   490.2  704.49     549  701.53   578.4   699.4
#Mann= 3 , 0 , 0
       0      .1       0   285.4    .045       0   345.4      .1       0
Bank Sta=285.4,345.4
XS Rating Curve= 0 ,0
Exp/Cntr=0.3,0.1

Type RM Length L Ch R = 1 ,68035.3 ,729,664,599.8
XS GIS Cut Line= 2
     1739860.596      595992.243     1738826.896      595781.887
#Sta/Elev= 30
       0  852.09    87.9   841.7   117.2  837.25   146.5  831.13   185.6  821.34
   195.4  818.02   214.9  809.93   234.4  801.07   273.5  781.94   332.1  752.39
   390.7  724.22     420  708.71   449.3  691.31   459.1  685.94   498.1  665.84
   527.4  652.37   566.5  637.77     586  632.43   595.8  631.11   605.6  631.12
   615.4  632.57     637   638.9   644.6  640.08   654.4   640.8   732.6  645.63
   761.9  647.02   800.9  648.08   830.2  649.62   957.2  665.68  1054.9  675.13
#Mann= 3 , 0 , 0
       0      .1       0   566.5    .045       0     637     .08       0
Bank Sta=566.5,637
XS Rating Curve= 0 ,0
Exp/Cntr=0.3,0.1

Type RM Length L Ch R = 1 ,67371.3 ,324.3,318.8,313.4
XS GIS Cut Line= 2
     1739011.555      594999.267     1738736.379      595855.112
#Sta/Elev= 30
       0  846.35    39.1  837.26    58.6  832.29    78.2  826.62      88  822.94
    97.7  818.49   166.1  785.58   254.1  743.53   302.9  721.08   312.7  715.97
     342  698.65   371.3  682.11   439.7  645.93   453.1  639.48   459.3  636.54
     469  632.31   478.8  630.84   488.6   631.6   508.1  637.51   517.9  639.05
   527.7  639.59   566.8  640.46   586.3  641.21   693.8  646.84   703.6  647.96
   713.3  650.23   742.6  659.41   781.7  672.29   850.1  695.42     899  711.62
#Mann= 3 , 0 , 0
       0      .1       0   453.1    .045       0   517.9     .06       0
Bank Sta=453.1,517.9
XS Rating Curve= 0 ,0
Exp/Cntr=0.3,0.1

Type RM Length L Ch R = 1 ,67052.5 ,302.8,317.7,332.6
XS GIS Cut Line= 3
     1738612.075      595127.041     1738499.576      595700.212
      1738195.65       596129.85
#Sta/Elev= 30
       0  740.74    48.7  724.13    68.2  716.02    87.6  706.28   116.8  687.97
   155.8   658.9   175.2   645.4   191.1   637.4   204.4  632.49   214.2  630.87
   223.9  630.88   243.4  636.02   251.1  637.08   418.6  641.77   447.8  643.39
   525.7  661.26   574.4  671.26   623.1  684.78   632.8  686.18   671.8  688.78
   710.8  696.22   759.5  698.48   847.2  705.71     857  705.78     896  702.95
   905.7  703.48     935  708.91   964.2  711.84  1022.7  715.07  1110.4   716.9
#Mann= 3 , 0 , 0
       0      .1       0   191.1    .045       0   251.1     .06       0
Bank Sta=191.1,251.1
XS Rating Curve= 0 ,0
Exp/Cntr=0.3,0.1

Type RM Length L Ch R = 1 ,66734.8 ,339.3,380.8,422.2
XS GIS Cut Line= 2
     1738356.037      595106.905     1737977.245      595769.525
#Sta/Elev= 30
       0  681.57    58.7  675.41    97.8  673.03   107.6  671.55   117.4  667.34
   146.8  647.21   165.3  635.96   176.1  631.36   185.9  630.46   195.7  631.19
   205.5  632.76   215.3  634.08   234.8  635.11   264.2  635.63   332.7  635.99
   381.6  637.56   401.2  638.74   430.6  641.12   450.1  643.38   469.7  646.53
   489.3  650.36     499   652.8   508.8  656.14   596.9  689.87   626.3  700.49
   655.6  710.56   733.9  736.34   743.7  739.14   753.5  740.69   763.2  740.25
#Mann= 3 , 0 , 0
       0      .1       0   165.3    .045       0   205.5     .06       0
Bank Sta=165.3,205.5
XS Rating Curve= 0 ,0
Exp/Cntr=0.3,0.1

Type RM Length L Ch R = 1 ,66353.9 ,335,371.6,408.4
XS GIS Cut Line= 2
      1738548.38      595030.268     1737620.446      595160.943
#Sta/Elev= 30
       0  741.64    58.6  728.29   107.4  715.06   117.1  711.84   126.9  707.93
   136.7  703.32   156.2  692.78   165.9  688.35   175.7  685.06   195.2  679.68
   224.5  672.51   292.8  658.54   370.9  649.14   380.7  648.31   429.5  645.55
   527.1   638.2   585.7  635.75     601  632.87     615  630.04   624.7  629.24
   634.5  629.91   644.2  632.72     661     641   693.1  656.73   732.1  676.78
   829.7   729.7   868.8  753.35   907.8  773.94   927.3  783.61   937.1  787.98
#Mann= 3 , 0 , 0
       0     .06       0     601    .045       0     661      .1       0
Bank Sta=601,661
XS Rating Curve= 0 ,0
Exp/Cntr=0.3,0.1

Type RM Length L Ch R = 1 ,65982.3 ,248.3,245.9,243.4
XS GIS Cut Line= 2
     1738353.631      594999.387     1737736.426      594511.579
#Sta/Elev= 30
       0   675.8      59  660.75     118  646.55   127.8  644.54   137.7  643.24
   206.5  638.03   273.8  633.62   285.2  631.97     295  629.44   304.8  628.09
   314.7  628.69   324.5  632.47   333.8   638.4   344.2  644.75   383.5  667.22
   422.8  690.49   442.5  701.66   452.4  706.98   462.2  712.08   511.4  736.33
   521.2  740.86     531  743.92   550.7  748.31   560.5  749.54   570.4  750.25
   599.9   750.6   629.4  749.93   658.9  748.46   737.5  743.16   786.7  741.94
#Mann= 3 , 0 , 0
       0     .06       0   273.8    .045       0   333.8      .1       0
Bank Sta=273.8,333.8
XS Rating Curve= 0 ,0
Exp/Cntr=0.3,0.1

Type RM Length L Ch R = 1 ,65736.4 ,246.3,232.4,214.7
XS GIS Cut Line= 2
     1738747.162      594957.988     1738093.435      594496.333
#Sta/Elev= 30
       0  802.14     9.8  797.07    19.5  792.72      39  785.81    68.3  776.68
   107.4  766.18   165.9  752.41   195.2  745.02   224.5  736.78   234.2  733.85
     244  730.34   273.3  718.05   302.6  705.15   390.4   664.6   429.4  647.54
   439.2  643.82     449  641.29   468.5  638.56   478.2  637.63   517.3  635.42
   545.4  632.78   556.3   630.7   566.1  628.26   575.8  627.11   585.6  628.27
   605.4  635.56   634.4  643.82   712.5  664.92   790.5  687.32   800.3  689.38
#Mann= 3 , 0 , 0
       0     .06       0   545.4    .045       0   605.4     .06       0
Bank Sta=545.4,605.4
XS Rating Curve= 0 ,0
Exp/Cntr=0.3,0.1

Type RM Length L Ch R = 1 ,65504   ,102.5,99.2,99
XS GIS Cut Line= 4
     1738928.117      594669.757     1738429.269      594437.482
      1738348.14      594419.036     1738057.957      594465.272
#Sta/Elev= 30
       0   813.2    49.1  794.75    68.8  786.59   108.1  769.19   127.7  761.55
   147.4  754.56   176.9  745.33   196.5  740.21     226  736.12   235.8   733.4
   265.3  721.01   304.6  703.39   422.5  648.03   432.4  643.79   442.2  641.05
     452   639.8   520.8  635.74   540.4  633.91   547.7  632.74   568.8  627.84
     578  627.01   587.2  627.62   607.7  632.34     615  633.75     751  653.77
   780.4  660.83   819.6  668.26   858.8     678   897.9  684.53   927.3  690.22
#Mann= 3 , 0 , 0
       0     .06       0   547.7    .045       0   607.7     .06       0
Bank Sta=547.7,607.7
XS Rating Curve= 0 ,0
Exp/Cntr=0.3,0.1

Type RM Length L Ch R = 1 ,65404.8 ,613.6,541.8,470.4
XS GIS Cut Line= 5
      1739183.38      594173.628     1738719.106      594463.833
     1738461.322      594343.803     1738351.426      594318.817
     1738042.466      594368.044
#Sta/Elev= 30
       0  677.56    19.6  676.35    29.3  678.51    68.4  691.47      88   696.3
   117.3  701.08   136.9  702.48   205.3  700.71   273.8  695.96   312.9  694.23
   410.6  695.84   430.2  695.47   498.6  690.94   537.7  690.23   547.5  690.85
     675   642.7   694.6  636.68   704.4  635.03     724  633.68   792.6  633.39
   847.9  628.59   869.4   626.9   888.2  627.24   907.9  631.62   935.2  634.07
   993.4  636.31  1042.3  640.31  1149.9  655.61  1198.8  659.65  1257.4  669.38
#Mann= 3 , 0 , 0
       0     .08       0   847.9    .045       0   907.9     .06       0
Bank Sta=847.9,907.9
XS Rating Curve= 0 ,0
Exp/Cntr=0.3,0.1
